--- ExtranTestImport.prj (project) ---

Proj Title=SWMM Extran Tests Circular
Current Plan=p01
Default Exp/Contr=0.3,0.1
English Units
Geom File=g02
Geom File=g07
Geom File=g01
Geom File=g04
Unsteady File=u01
Unsteady File=u02
Unsteady File=u03
Unsteady File=u04
Unsteady File=u06
Unsteady File=u07
Unsteady File=u08
Plan File=p06
Plan File=p01
Plan File=p02
Plan File=p03
Plan File=p04
Y Axis Title=Elevation
X Axis Title(PF)=Main Channel Distance
X Axis Title(XS)=Station
BEGIN DESCRIPTION:
END DESCRIPTION:
DSS File=.\SWMM Extran Datasets\EXTRAN 7 Example.dss
DSS File=dss
DSS Export Rating Curves= 0
DSS Export Rating Curve Sorted= 0
DSS Export Volume Flow Curves= 0
DXF OffsetX= 0
DXF OffsetY= 0
DXF ScaleX= 1
DXF ScaleY= 10

--- ExtranTestImport.p01 (plan) ---

Plan Title=Extran7 - Pump
Program Version=7.01
Short Identifier=Extran7 - Pump
Simulation Date=01Jan1988,0000,01Jan1988,0600
Geom File=g07
Flow File=u03
Subcritical Flow
K Sum by GR= 0
Std Step Tol= 0.01
Critical Tol= 0.01
Num of Std Step Trials= 20
Max Error Tol= 0.3
Flow Tol Ratio= 0.001
Split Flow NTrial= 30
Split Flow Tol= 0.02
Split Flow Ratio= 0.02
Log Output Level= 0
Friction Slope Method= 1
Unsteady Friction Slope Method= 2
Unsteady Bridges Friction Slope Method= 1
Parabolic Critical Depth
Global Vel Dist= 0 , 0 , 0
Global Log Level= 0
CheckData=True
Encroach Param=-1 ,0,0, 0
Flow Ratio Tolerance=0.1
Flow Ratio Min Ratio=0.5
Flow Ratio Max Ratio=4
Flow Ratio Max Iterations= 10
Computation Interval=10SEC
Output Interval=5MIN
Instantaneous Interval=1HOUR
Mapping Interval=5MIN
Computation Time Step Use Courant=        0
Computation Time Step Use Time Series=    0
Computation Time Step Count To Double=0
Computation Time Step Max Doubling=0
Computation Time Step Max Halving=0
Computation Time Step Residence Courant=0
Computation Time Step TS=, 0
Computation Time Step TS=, 0
Computation Time Step TS=, 0
Computation Time Step TS=, 0
Computation Time Step TS=, 0
Computation Time Step TS=, 0
Computation Time Step TS=, 0
Computation Time Step TS=, 0
Computation Time Step TS=, 0
Computation Time Step TS=, 0
Computation Time Step TS=, 0
Computation Time Step TS=, 0
Computation Time Step TS=, 0
Computation Time Step TS=, 0
Computation Time Step TS=, 0
Computation Time Step TS=, 0
Computation Time Step TS=, 0
Computation Time Step TS=, 0
Computation Time Step TS=, 0
Computation Time Step TS=, 0
Computation Time Step TS=, 0
Computation Time Step TS=, 0
Computation Time Step TS=, 0
Computation Time Step TS=, 0
Computation Time Step TS=, 0
Computation Time Step TS=, 0
Computation Time Step TS=, 0
Computation Time Step TS=, 0
Computation Time Step TS=, 0
Computation Time Step TS=, 0
Computation Time Step TS=, 0
Computation Time Step TS=, 0
Computation Time Step TS=, 0
Computation Time Step TS=, 0
Computation Time Step TS=, 0
Computation Time Step TS=, 0
Computation Time Step TS=, 0
Computation Time Step TS=, 0
Computation Time Step TS=, 0
Computation Time Step TS=, 0
Computation Time Step TS=, 0
Computation Time Step TS=, 0
Computation Time Step TS=, 0
Computation Time Step TS=, 0
Computation Time Step TS=, 0
Computation Time Step TS=, 0
Computation Time Step TS=, 0
Computation Time Step TS=, 0
Computation Time Step TS=, 0
Computation Time Step TS=, 0
Run HTab=-1
Run UNet=-1
Run Sediment= 0
Run PostProcess= 0
Run WQNet= 0
Run RASMapper= 0
UNET Theta= 1
UNET Theta Warmup= 1
UNET ZTol= 0.02
UNET ZSATol= 0.02
UNET MxIter= 20
UNET Max Iter WO Improvement= 0
UNET MaxInSteps= 0
UNET DtIC= 0
UNET DtMin= 0
UNET MaxCRTS= 20
UNET WFStab= 2
UNET SFStab= 1
UNET WFX= 1
UNET SFX= 1
UNET Gravity=32.17405
UNET 1D Methodology=Finite Difference
UNET DSS MLevel= 4
UNET Pardiso=0
UNET DZMax Abort= 100
UNET Use Existing IB Tables=-1
UNET Froude Reduction=False
UNET Froude Limit= 0.8
UNET Froude Power= 4
UNET D1 Cores= 0
UNET WindReference=Eulerian
UNET WindDragFormulation=Hsu (1988)
UNET D2 Coriolis=0
UNET D2 Cores= 0
UNET D2 Theta= 1
UNET D2 Theta Warmup= 1
UNET D2 Z Tol= 0.01
UNET D2 Volume Tol= 0.01
UNET D2 Max Iterations= 20
UNET D2 Advanced Convergence=0
UNET D2 WS Max Tol=0.15
UNET D2 WS RMS Tol=0.002
UNET D2 WS Stall Tol=1
UNET D2 Equation= 0
UNET D2 RampUpFraction=0.1
UNET D2 TimeSlices= 1
UNET D2 Turbulence Formulation=None
UNET D2 Eddy Viscosity=0.3
UNET D2 Transverse Eddy Viscosity=0.1
UNET D2 Smagorinsky Mixing=0.05
UNET D2 BCVolumeCheck=0
UNET D2 Cores=0
UNET D2 SolverType=PARDISO (Direct)
UNET D2 Minimum Iterations= 3
UNET D2 Maximum Iterations= 30
UNET D2 Restart Number= 10
UNET D2 Relaxation Coeff=1.3
UNET D2 SOR Precondition Iterations= 10
UNET D2 ILUT Maximum Fill= 8
UNET D2 ILUT Tolerance=1E-08
UNET D2 Convergence Tolerance=0.00001
Secondary Flow Approach=None
Spiral Intensity Factor=1
Spiral Intensity Adaptation Factor=1
Spiral Intensity Diffusion Factor=1
Momentum Dispersion Factor=1
Flow Smoothing Iterations=10
UNET D2 Name=Perimeter 1
UNET D2 Theta= 1
UNET D2 Theta Warmup= 1
UNET D2 Z Tol= 0.01
UNET D2 Volume Tol= 0.01
UNET D2 Max Iterations= 20
UNET D2 Advanced Convergence=0
UNET D2 WS Max Tol=0.15
UNET D2 WS RMS Tol=0.002
UNET D2 WS Stall Tol=1
UNET D2 Equation= 0
UNET D2 RampUpFraction=0.1
UNET D2 TimeSlices= 1
UNET D2 Turbulence Formulation=None
UNET D2 Eddy Viscosity=0.3
UNET D2 Transverse Eddy Viscosity=0.1
UNET D2 Smagorinsky Mixing=0.05
UNET D2 BCVolumeCheck=0
UNET D2 Cores=0
UNET D2 SolverType=PARDISO (Direct)
UNET D2 Minimum Iterations= 3
UNET D2 Maximum Iterations= 30
UNET D2 Restart Number= 10
UNET D2 Relaxation Coeff=1.3
UNET D2 SOR Precondition Iterations= 10
UNET D2 ILUT Maximum Fill= 0
UNET D2 ILUT Tolerance=0
UNET D2 Convergence Tolerance=0.00001
Secondary Flow Approach=None
Spiral Intensity Factor=1
Spiral Intensity Adaptation Factor=1
Spiral Intensity Diffusion Factor=1
Momentum Dispersion Factor=1
Flow Smoothing Iterations=10
PS Theta= 1
PS WS Tol= 0.01
PS Volume Tol= 0.01
PS Max Iterations= 20
PS Equation= 0
PS Advance Time Step=-1
PS Target Courant=0.9
PS Time Slices= 1
PS Iterate With 2D=0
PS Project Initial WSE from DS=-1
PS Ramp Up Initial WSE from US=-1
PS Cores=0
PS Name=Base
PS Theta= 1
PS WS Tol= 0.01
PS Volume Tol= 0.01
PS Max Iterations= 20
PS Equation= 1
PS Advance Time Step=-1
PS Target Courant=0.9
PS Time Slices= 1
PS Iterate With 2D=0
PS Project Initial WSE from DS=-1
PS Ramp Up Initial WSE from US=-1
PS Cores=0
UNET D1D2 MaxIter= 0
UNET D1D2 ZTol=0.01
UNET D1D2 QTol=0.1
UNET D1D2 MinQTol=1
DSS File=dss
Write IC File= 0
Write IC File at Fixed DateTime=0
Write IC File at Sim End=0
Echo Input=False
Echo Parameters=False
Echo Output=False
Write Detailed= 1
HDF Write Warmup=0
HDF Write Time Slices=0
HDF Flush=0
HDF Compression= 1
HDF Chunk Size= 1
HDF Spatial Parts= 1
HDF Use Max Rows=0
HDF Fixed Rows= 1
Calibration Method= 0
Calibration Iterations= 20
Calibration Max Change=0.05
Calibration Tolerance=0.2
Calibration Maximum=1.5
Calibration Minimum=0.5
Calibration Optimization Method= 1
WQ AD Non Conservative
WQ ULTIMATE=-1
WQ Max Comp Step=1HOUR
WQ Kinetics Update Frequency= 0
WQ Output Interval=15MIN
WQ Output Selected Increments=0
WQ Pathway Output Fequency=0
WQ Create Restart=0
WQ Fixed Restart=0
WQ System Summary=0
WQ Write To DSS=0
Sorting and Armoring Iterations= 10
XS Update Threshold= 0.02
Bed Roughness Predictor= 0
Processes Affected by Predictor=Sediment Only
Hydraulics Update Threshold= 0.02
Energy Slope Method= 1
Volume Change Method= 1
Sediment Retention Method= 0
Sediment TS Multiplier= 1
Warm Up Method= 0
XS Weighting Method= 0
Number of US Weighted Cross Sections= 1
Number of DS Weighted Cross Sections= 1
Upstream XS Weight=0
Main XS Weight=1
Downstream XS Weight=0
Number of DS XS's Weighted with US Boundary= 1
Upstream Boundary Weight= 1
Weight of XSs Associated with US Boundary= 0
Number of US XS's Weighted with DS Boundary= 1
Downstream Boundary Weight= 0.5
Weight of XSs Associated with DS Boundary= 0.5
Percentile Method= 0
Sediment Output Level= 3
Mass or Volume Output= 0
Output Increment Type= 1
Profile and TS Output Increment= 1
Transport Output Increment 1
XS Output Flag= 0
XS Output Increment= 10
Read HDF5 Sediment Hotstart= 0
Sediment Hotstart Type= 0
Write Gradation File= 0
Read Gradation Hotstart= 0
Write HDF5 File= 1
Write Binary Output= 1
Write DSS Sediment File= 0
DSS Sediment Output Type= 1
SV Curve= 0
Specific Gage Flag= 0
Subcell Erosion Methods= 0
Subcell Deposition Methods= 0
Advection Scheme= 1
Matrix Solver= 0
Implicit Weighting Factor= 1
Maximum Outer Loop Convergence Iterations= 5
Convergence Maximum Absolute= 0.001
Convergence RMSE= 0.0001
Grain Fractions Max Abs Error= 0.001
Max Subgrid Regions= 1
Max Subgrid Length Scale= 3.402823E+38
Initial Layer Thickness= 3
Min Layer Thickness= 0.1
Max Layer Thickness= 6
Number of Layers= 5

--- ExtranTestImport.p02 (plan) ---

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Plan Title=Extran 2
Program Version=7.00
Short Identifier=Extran 2
Geom File=g02
Flow File=u04
BEGIN DESCRIPTION:
Geometry includes top inlets and 2D areas to allow flow to surcharge to the srface.
The observed data included in this dataset are SWMM results for the EXTRAN 2 test for comparison.
END DESCRIPTION:
Computation Interval=20SEC
Write Detailed= 0

--- ExtranTestImport.p03 (plan) ---

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Plan Title=Extran 4 - Weir
Program Version=7.00
Short Identifier=Extran 4 - Weir
Geom File=g01
Flow File=u06
BEGIN DESCRIPTION:
Geometry includes top inlets and 2D areas to allow flow to surcharge to the srface.
The observed data included in this dataset are SWMM results for the EXTRAN 4 test for comparison.
END DESCRIPTION:
Computation Interval=20SEC
UNET D2 Name=Surface Stor 1
UNET D2 Name=Surface Stor 2
PS Cores=1
Write Detailed= 0

--- ExtranTestImport.p04 (plan) ---

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Plan Title=Extran 5 - Orifice
Program Version=7.00
Short Identifier=Extran 5 - Orifice
Geom File=g04
Flow File=u07
BEGIN DESCRIPTION:
Geometry includes top inlets and 2D areas to allow flow to surcharge to the srface.
The observed data included in this dataset are SWMM results for the EXTRAN 5 test for comparison.
END DESCRIPTION:
Computation Interval=20SEC
UNET D2 Name=Surface Stor 1
UNET D2 Name=Surface Stor 2
PS Target Courant=0.6
PS Cores=1
Write Detailed= 0

--- ExtranTestImport.p06 (plan) ---

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Plan Title=Extran 1
Program Version=7.00
Short Identifier=Extran 1
Geom File=g02
Flow File=u01
BEGIN DESCRIPTION:
Geometry includes top inlets and 2D areas to allow flow to surcharge to the srface.
The observed data included in this dataset are SWMM results for the EXTRAN 1 test for comparison.
END DESCRIPTION:
UNET D2 Name=Surface Stor 1
UNET D2 Name=Surface Stor 2
Write Detailed= 0

--- ExtranTestImport.u03 (unsteady flow) ---

Flow Title=Extran7 -InlinePump
Program Version=7.00
Use Restart= 0
Initial Storage Elev=Perimeter 1     ,94.4,0
Boundary Location=                ,                ,        ,        ,                ,Perimeter 1     ,                ,DS Boundary                     ,                                ,
Friction Slope=0.0035
Boundary Location=                ,                ,        ,        ,                ,                ,                ,                                ,Base [81009]                    ,
Interval=15MIN
Flow Hydrograph= 49
       0      50      50      50      50      50      50      50      50      50
      50      50      50       0       0       0       0       0       0       0
       0       0       0       0       0       0       0       0       0       0
       0       0       0       0       0       0       0       0       0       0
       0       0       0       0       0       0       0       0       0
Stage Hydrograph TW Check=0
Use DSS=False
Use Fixed Start Time=False
Is Critical Boundary=False
Boundary Location=                ,                ,        ,        ,                ,                ,                ,                                ,Base [82309]                    ,
Interval=15MIN
Flow Hydrograph= 49
       0      40      40      40      40      40      40      40      40      40
      40      40      40       0       0       0       0       0       0       0
       0       0       0       0       0       0       0       0       0       0
       0       0       0       0       0       0       0       0       0       0
       0       0       0       0       0       0       0       0       0
Stage Hydrograph TW Check=0
Use DSS=False
Use Fixed Start Time=False
Is Critical Boundary=False
Boundary Location=                ,                ,        ,        ,                ,                ,                ,                                ,Base [80408]                    ,
Interval=15MIN
Flow Hydrograph= 49
       0      45      45      45      45      45      45      45      45      45
      45      45      45       0       0       0       0       0       0       0
       0       0       0       0       0       0       0       0       0       0
       0       0       0       0       0       0       0       0       0       0
       0       0       0       0       0       0       0       0       0
Stage Hydrograph TW Check=0
Flow Hydrograph QMult= 0.5
Use DSS=False
Use Fixed Start Time=False
Is Critical Boundary=False
Boundary Location=                ,                ,        ,        ,                ,                ,Pump Station #1 ,                                ,                                ,
Rule Operation=Type=0,Var Type=1,Comment=Make a pump efficiency curve based on depth not head
Rule Operation=Type=1,Var Name=82309_Invert,Var Type=1,Real=112.2
Rule Operation=Type=2,Var Name=82309 WSEL,Var Type=1,PipeNode=Base [82309],Sim Group=Pipe Nodes,Sim Function=WS Elevation,Time=5,LBStart=0.16,LBEnd=0
Rule Operation=Type=0,Var Type=1,Comment=Compute the depth for the *cell*
Rule Operation=Type=5,Var Name=82309_Depth,Var Type=1,MathOperator1=2,MathOperator2=0,MathOperator3=0
Rule Expression=,Variable=82309 WSEL
Rule Expression=,Variable=82309_Invert
Rule Operation=Type=0,Var Type=1,Comment=Get the Pump Flow From the Table
Rule Operation=Type=6,Var Name=Table Pump Flow,Var Type=1,TableMode=3,Table2D=0,TableArgX=82309 Depth,TableArgY=
Rule Expression=,Variable=82309_Depth
Rule Table=6,1
       1       5       7      25    42.6    42.7
       5       5      10      20      20      20
Rule Operation=Type=0,Var Type=1,Comment=Set the pump flow from the table
Rule Operation=Type=4,Var Type=1,Branch Type=0,Branch Or=0,BranchCompare1=4,BranchCompare2=0
Rule Expression=,Variable=82309_Depth
Rule Expression=,Constant=0.5
Rule Operation=Type=3,Var Type=1,PumpGroup=Group #1,PumpName=Pump #1,Sim Group=Pump Stations,Sim Function=Turn Pump On
Rule Operation=Type=3,Var Type=1,PumpGroup=Group #1,PumpName=Pump #1,Sim Group=Pump Stations,Sim Function=Station.Pump Flow
Rule Expression=,Variable=Table Pump Flow
Rule Operation=Type=4,Var Type=1,Branch Type=4,Branch Or=0,BranchCompare1=0,BranchCompare2=0
Rule Operation=Type=3,Var Type=1,PumpGroup=Group #1,PumpName=Pump #1,Sim Group=Pump Stations,Sim Function=Turn Pump Off
Rule Operation=Type=4,Var Type=1,Branch Type=5,Branch Or=0,BranchCompare1=0,BranchCompare2=0
Precipitation Mode=Disable
Wind Mode=No Wind Forces
Wave Mode=No Wave Forcing
Met BC=Precipitation|Expanded View=0
Met BC=Precipitation|Point Interpolation=Nearest
Met BC=Precipitation|Gridded Source=DSS
Met BC=Precipitation|Gridded Interpolation=
Met BC=Evapotranspiration|Expanded View=0
Met BC=Evapotranspiration|Point Interpolation=Nearest
Met BC=Evapotranspiration|Gridded Source=DSS
Met BC=Evapotranspiration|Gridded Interpolation=
Met BC=Wind Speed|Expanded View=0
Met BC=Wind Speed|Point Interpolation=Nearest
Met BC=Wind Speed|Gridded Source=DSS
Met BC=Wind Speed|Gridded Interpolation=
Met BC=Wind Direction|Expanded View=0
Met BC=Wind Direction|Point Interpolation=Nearest
Met BC=Wind Direction|Gridded Source=DSS
Met BC=Wind Direction|Gridded Interpolation=
Met BC=Wind Velocity X|Expanded View=0
Met BC=Wind Velocity X|Point Interpolation=Nearest
Met BC=Wind Velocity X|Gridded Source=DSS
Met BC=Wind Velocity X|Gridded Interpolation=
Met BC=Wind Velocity Y|Expanded View=0
Met BC=Wind Velocity Y|Point Interpolation=Nearest
Met BC=Wind Velocity Y|Gridded Source=DSS
Met BC=Wind Velocity Y|Gridded Interpolation=
Met BC=Wave Forcing X|Expanded View=0
Met BC=Wave Forcing X|Point Interpolation=Nearest
Met BC=Wave Forcing X|Gridded Source=DSS
Met BC=Wave Forcing X|Gridded Interpolation=
Met BC=Wave Forcing Y|Expanded View=0
Met BC=Wave Forcing Y|Point Interpolation=Nearest
Met BC=Wave Forcing Y|Gridded Source=DSS
Met BC=Wave Forcing Y|Gridded Interpolation=
Met BC=Air Density|Mode=Constant
Met BC=Air Density|Expanded View=0
Met BC=Air Density|Constant Value=1.225
Met BC=Air Density|Constant Units=kg/m3
Met BC=Air Density|Point Interpolation=Nearest
Met BC=Air Density|Gridded Source=DSS
Met BC=Air Density|Gridded Interpolation=
Met BC=Air Temperature|Expanded View=0
Met BC=Air Temperature|Point Interpolation=Nearest
Met BC=Air Temperature|Gridded Source=DSS
Met BC=Air Temperature|Gridded Interpolation=
Met BC=Humidity|Expanded View=0
Met BC=Humidity|Point Interpolation=Nearest
Met BC=Humidity|Gridded Source=DSS
Met BC=Humidity|Gridded Interpolation=
Met BC=Air Pressure|Mode=Constant
Met BC=Air Pressure|Expanded View=0
Met BC=Air Pressure|Constant Value=1013.2
Met BC=Air Pressure|Constant Units=mb
Met BC=Air Pressure|Point Interpolation=
Met BC=Air Pressure|Gridded Source=DSS
Met BC=Air Pressure|Gridded Interpolation=
Observed Time Series=Stage|TS Name=BC Line: DS Boundary
Observed Time Series=Stage|TS Used=-1
Observed Time Series=Stage|TS Source=DSS
Observed Time Series=Stage|TS DSS Filename=.\SWMM Extran Datasets\EXTRAN 7 example.dss
Observed Time Series=Stage|TS DSS Pathname=/Base/10208/Stage/31Dec1987-01Jan1988/5Minute/EXTRAN 7 example/
Observed Time Series=Stage|TS Table Mode=0
Observed Time Series=Stage|TS Table Use Fixed Start=0
Observed Time Series=Stage|TS Table StartDateTime=01Jan1988 00:00:00
Observed Time Series=Stage|TS Table Interval=1 Hour
Observed Time Series=Stage|TS Table Data Units=ft
Observed Time Series=Stage|TS Table Data Type=INST-VAL
Observed Time Series=Stage|TS Constant Units=ft
Observed Time Series=Stage|TS Name=Pipe Node: Base [15009]
Observed Time Series=Stage|TS Used=-1
Observed Time Series=Stage|TS Source=DSS
Observed Time Series=Stage|TS DSS Filename=.\SWMM Extran Datasets\EXTRAN 7 example.dss
Observed Time Series=Stage|TS DSS Pathname=/Base/15009/Stage//5Minute/EXTRAN 7 example/
Observed Time Series=Stage|TS Table Mode=0
Observed Time Series=Stage|TS Table Use Fixed Start=0
Observed Time Series=Stage|TS Table StartDateTime=01Jan1988 00:00:00
Observed Time Series=Stage|TS Table Interval=1 Hour
Observed Time Series=Stage|TS Name=Pipe Node: Base [81309]
Observed Time Series=Stage|TS Used=-1
Observed Time Series=Stage|TS Source=DSS
Observed Time Series=Stage|TS DSS Filename=.\SWMM Extran Datasets\EXTRAN 7 example.dss
Observed Time Series=Stage|TS DSS Pathname=/Base/81309/Stage//5Minute/EXTRAN 7 example/
Observed Time Series=Stage|TS Table Mode=0
Observed Time Series=Stage|TS Table Use Fixed Start=0
Observed Time Series=Stage|TS Table Interval=1 Hour
Observed Time Series=Stage|TS Name=Pipe Node: Base [81009]
Observed Time Series=Stage|TS Used=-1
Observed Time Series=Stage|TS Source=DSS
Observed Time Series=Stage|TS DSS Filename=.\SWMM Extran Datasets\EXTRAN 7 example.dss
Observed Time Series=Stage|TS DSS Pathname=/Base/81009/Stage//5Minute/EXTRAN 7 example/
Observed Time Series=Stage|TS Table Mode=0
Observed Time Series=Stage|TS Table Use Fixed Start=0
Observed Time Series=Stage|TS Table Interval=1 Hour
Observed Time Series=Stage|TS Name=Pipe Node: Base [16109]
Observed Time Series=Stage|TS Used=-1
Observed Time Series=Stage|TS Source=DSS
Observed Time Series=Stage|TS DSS Filename=.\SWMM Extran Datasets\EXTRAN 7 example.dss
Observed Time Series=Stage|TS DSS Pathname=/Base/16109/Stage//5Minute/EXTRAN 7 example/
Observed Time Series=Stage|TS Table Mode=0
Observed Time Series=Stage|TS Table Use Fixed Start=0
Observed Time Series=Stage|TS Table StartDateTime=01Jan1988 00:00:00
Observed Time Series=Stage|TS Table Interval=1 Hour
Observed Time Series=Stage|TS Table Data Units=ft
Observed Time Series=Stage|TS Table Data Type=INST-VAL
Observed Time Series=Stage|TS Constant Units=ft
Observed Time Series=Stage|TS Name=Pipe Node: Base [82309]
Observed Time Series=Stage|TS Used=-1
Observed Time Series=Stage|TS Source=DSS
Observed Time Series=Stage|TS DSS Filename=.\SWMM Extran Datasets\EXTRAN 7 example.dss
Observed Time Series=Stage|TS DSS Pathname=/Base/82309/Stage//5Minute/EXTRAN 7 example/
Observed Time Series=Stage|TS Table Mode=0
Observed Time Series=Stage|TS Table Use Fixed Start=0
Observed Time Series=Stage|TS Table Interval=1 Hour
Observed Time Series=Stage|TS Name=Pipe Node: Base [80608]
Observed Time Series=Stage|TS Used=-1
Observed Time Series=Stage|TS Source=DSS
Observed Time Series=Stage|TS DSS Filename=.\SWMM Extran Datasets\EXTRAN 7 example.dss
Observed Time Series=Stage|TS DSS Pathname=/Base/80608/Stage//5Minute/EXTRAN 7 example/
Observed Time Series=Stage|TS Table Mode=0
Observed Time Series=Stage|TS Table Use Fixed Start=0
Observed Time Series=Stage|TS Table Interval=1 Hour
Observed Time Series=Stage|TS Name=Pipe Node: Base [80408]
Observed Time Series=Stage|TS Used=-1
Observed Time Series=Stage|TS Source=DSS
Observed Time Series=Stage|TS DSS Filename=.\SWMM Extran Datasets\EXTRAN 7 example.dss
Observed Time Series=Stage|TS DSS Pathname=/Base/80408/Stage//5Minute/EXTRAN 7 example/
Observed Time Series=Stage|TS Table Mode=0
Observed Time Series=Stage|TS Table Use Fixed Start=0
Observed Time Series=Stage|TS Table Interval=1 Hour
Observed Time Series=Stage|TS Name=Pipe Node: Base [16009]
Observed Time Series=Stage|TS Used=-1
Observed Time Series=Stage|TS Source=DSS
Observed Time Series=Stage|TS DSS Filename=.\SWMM Extran Datasets\EXTRAN 7 example.dss
Observed Time Series=Stage|TS DSS Pathname=/Base/16009/Stage//5Minute/EXTRAN 7 example/
Observed Time Series=Stage|TS Table Mode=0
Observed Time Series=Stage|TS Table Use Fixed Start=0
Observed Time Series=Stage|TS Table Interval=1 Hour
Observed Time Series=Flow|TS Name=BC Line: DS Boundary
Observed Time Series=Flow|TS Used=-1
Observed Time Series=Flow|TS Source=DSS
Observed Time Series=Flow|TS DSS Filename=.\SWMM Extran Datasets\EXTRAN 7 Example.dss
Observed Time Series=Flow|TS DSS Pathname=/Base/10208/Flow/31Dec1987-01Jan1988/5Minute/EXTRAN 7 example/
Observed Time Series=Flow|TS Table Mode=0
Observed Time Series=Flow|TS Table Use Fixed Start=0
Observed Time Series=Flow|TS Table StartDateTime=01Jan1988 00:00:00
Observed Time Series=Flow|TS Table Interval=1 Hour
Observed Time Series=Flow|TS Table Data Units=cfs
Observed Time Series=Flow|TS Table Data Type=INST-VAL
Observed Time Series=Flow|TS Constant Units=cfs
Observed Time Series=Flow|TS Name=Pipe Node: Base [15009]
Observed Time Series=Flow|TS Used=-1
Observed Time Series=Flow|TS Source=DSS
Observed Time Series=Flow|TS DSS Filename=.\SWMM Extran Datasets\EXTRAN 7 example.dss
Observed Time Series=Flow|TS DSS Pathname=/Base/15009/Flow//5Minute/EXTRAN 7 example/
Observed Time Series=Flow|TS Table Mode=0
Observed Time Series=Flow|TS Table Use Fixed Start=0
Observed Time Series=Flow|TS Table StartDateTime=01Jan1988 00:00:00
Observed Time Series=Flow|TS Table Interval=1 Hour
Observed Time Series=Flow|TS Table Data Units=cfs
Observed Time Series=Flow|TS Constant Units=cfs
Observed Time Series=Flow|TS Name=Pipe Node: Base [81309]
Observed Time Series=Flow|TS Used=-1
Observed Time Series=Flow|TS Source=DSS
Observed Time Series=Flow|TS DSS Filename=.\SWMM Extran Datasets\EXTRAN 7 example.dss
Observed Time Series=Flow|TS DSS Pathname=/Base/81309/Flow//5Minute/EXTRAN 7 example/
Observed Time Series=Flow|TS Table Mode=0
Observed Time Series=Flow|TS Table Use Fixed Start=0
Observed Time Series=Flow|TS Table StartDateTime=01Jan1988 00:00:00
Observed Time Series=Flow|TS Table Interval=1 Hour
Observed Time Series=Flow|TS Table Data Units=cfs
Observed Time Series=Flow|TS Constant Units=cfs
Observed Time Series=Flow|TS Name=Pipe Node: Base [81009]
Observed Time Series=Flow|TS Used=-1
Observed Time Series=Flow|TS Source=DSS
Observed Time Series=Flow|TS DSS Filename=.\SWMM Extran Datasets\EXTRAN 7 example.dss
Observed Time Series=Flow|TS DSS Pathname=/Base/81009/Flow//5Minute/EXTRAN 7 example/
Observed Time Series=Flow|TS Table Mode=0
Observed Time Series=Flow|TS Table Use Fixed Start=0
Observed Time Series=Flow|TS Table StartDateTime=01Jan1988 00:00:00
Observed Time Series=Flow|TS Table Interval=1 Hour
Observed Time Series=Flow|TS Table Data Units=cfs
Observed Time Series=Flow|TS Constant Units=cfs
Observed Time Series=Flow|TS Name=Pipe Node: Base [16109]
Observed Time Series=Flow|TS Used=-1
Observed Time Series=Flow|TS Source=DSS
Observed Time Series=Flow|TS DSS Filename=.\SWMM Extran Datasets\EXTRAN 7 example.dss
Observed Time Series=Flow|TS DSS Pathname=/Base/16109/Flow//5Minute/EXTRAN 7 example/
Observed Time Series=Flow|TS Table Mode=0
Observed Time Series=Flow|TS Table Use Fixed Start=0
Observed Time Series=Flow|TS Table StartDateTime=01Jan1988 00:00:00
Observed Time Series=Flow|TS Table Interval=1 Hour
Observed Time Series=Flow|TS Table Data Units=cfs
Observed Time Series=Flow|TS Table Data Type=INST-VAL
Observed Time Series=Flow|TS Constant Units=cfs
Observed Time Series=Flow|TS Name=Pipe Node: Base [82309]
Observed Time Series=Flow|TS Used=-1
Observed Time Series=Flow|TS Source=DSS
Observed Time Series=Flow|TS DSS Filename=.\SWMM Extran Datasets\EXTRAN 7 example.dss
Observed Time Series=Flow|TS DSS Pathname=/Base/82309/Flow//5Minute/EXTRAN 7 example/
Observed Time Series=Flow|TS Table Mode=0
Observed Time Series=Flow|TS Table Use Fixed Start=0
Observed Time Series=Flow|TS Table StartDateTime=01Jan1988 00:00:00
Observed Time Series=Flow|TS Table Interval=1 Hour
Observed Time Series=Flow|TS Table Data Units=cfs
Observed Time Series=Flow|TS Constant Units=cfs
Observed Time Series=Flow|TS Name=Pipe Node: Base [80608]
Observed Time Series=Flow|TS Used=-1
Observed Time Series=Flow|TS Source=DSS
Observed Time Series=Flow|TS DSS Filename=.\SWMM Extran Datasets\EXTRAN 7 example.dss
Observed Time Series=Flow|TS DSS Pathname=/Base/80608/Flow//5Minute/EXTRAN 7 example/
Observed Time Series=Flow|TS Table Mode=0
Observed Time Series=Flow|TS Table Use Fixed Start=0
Observed Time Series=Flow|TS Table StartDateTime=01Jan1988 00:00:00
Observed Time Series=Flow|TS Table Interval=1 Hour
Observed Time Series=Flow|TS Table Data Units=cfs
Observed Time Series=Flow|TS Constant Units=cfs
Observed Time Series=Flow|TS Name=Pipe Node: Base [80408]
Observed Time Series=Flow|TS Used=-1
Observed Time Series=Flow|TS Source=DSS
Observed Time Series=Flow|TS DSS Filename=.\SWMM Extran Datasets\EXTRAN 7 example.dss
Observed Time Series=Flow|TS DSS Pathname=/Base/80408/Flow//5Minute/EXTRAN 7 example/
Observed Time Series=Flow|TS Table Mode=0
Observed Time Series=Flow|TS Table Use Fixed Start=0
Observed Time Series=Flow|TS Table StartDateTime=01Jan1988 00:00:00
Observed Time Series=Flow|TS Table Interval=1 Hour
Observed Time Series=Flow|TS Table Data Units=cfs
Observed Time Series=Flow|TS Constant Units=cfs
Observed Time Series=Flow|TS Name=Pipe Node: Base [16009]
Observed Time Series=Flow|TS Used=-1
Observed Time Series=Flow|TS Source=DSS
Observed Time Series=Flow|TS DSS Filename=.\SWMM Extran Datasets\EXTRAN 7 example.dss
Observed Time Series=Flow|TS DSS Pathname=/Base/16009/Flow//5Minute/EXTRAN 7 example/
Observed Time Series=Flow|TS Table Mode=0
Observed Time Series=Flow|TS Table Use Fixed Start=0
Observed Time Series=Flow|TS Table StartDateTime=01Jan1988 00:00:00
Observed Time Series=Flow|TS Table Interval=1 Hour
Observed Time Series=Flow|TS Table Data Units=cfs
Observed Time Series=Flow|TS Table Data Type=INST-VAL
Observed Time Series=Flow|TS Constant Units=cfs
Non-Newtonian Method= 0 ,
Non-Newtonian Constant Vol Conc=0
Non-Newtonian Yield Method= 0 ,
Non-Newtonian Yield Coef=0, 0
User Yeild=   0
Non-Newtonian Sed Visc= 0 ,
Non-Newtonian Obrian B=0
User Viscosity=0
User Viscosity Ratio=0
Herschel-Bulkley Coef=0, 0
Clastic Method= 0 ,
Coulomb Phi=0
Voellmy X=0
Non-Newtonian Hindered FV= 0
Non-Newtonian FV K=0
Non-Newtonian ds=0
Non-Newtonian Max Cv=0
Non-Newtonian Bulking Method= 0 ,
Non-Newtonian High C Transport= 0 ,
Lava Activation= 0
Temperature=1300,15,,15,14,980
Heat Ballance=1,1200,0.5,1,70,0.95
Viscosity=1000,,,
Profile Coefficient=4,1.3,
Lava Param=,2500,

--- ExtranTestImport.u01 (unsteady flow) ---

Flow Title=Extran1
Program Version=7.00
Use Restart= 0
Boundary Location=                ,                ,        ,        ,                ,Perimeter 1     ,                ,DS Boundary                     ,                                ,
Friction Slope=0.0045
Boundary Location=                ,                ,        ,        ,                ,                ,                ,                                ,Base [81009]                    ,
Interval=15MIN
Flow Hydrograph= 49
       0      50      50      50      50      50      50      50      50      50
      50      50      50       0       0       0       0       0       0       0
       0       0       0       0       0       0       0       0       0       0
       0       0       0       0       0       0       0       0       0       0
       0       0       0       0       0       0       0       0       0
Stage Hydrograph TW Check=0
Use DSS=False
Use Fixed Start Time=False
Is Critical Boundary=False
Boundary Location=                ,                ,        ,        ,                ,                ,                ,                                ,Base [82309]                    ,
Interval=15MIN
Flow Hydrograph= 49
       0      40      40      40      40      40      40      40      40      40
      40      40      40       0       0       0       0       0       0       0
       0       0       0       0       0       0       0       0       0       0
       0       0       0       0       0       0       0       0       0       0
       0       0       0       0       0       0       0       0       0
Stage Hydrograph TW Check=0
Use DSS=False
Use Fixed Start Time=False
Is Critical Boundary=False
Boundary Location=                ,                ,        ,        ,                ,                ,                ,                                ,Base [80408]                    ,
Interval=15MIN
Flow Hydrograph= 49
       0      45      45      45      45      45      45      45      45      45
      45      45      45       0       0       0       0       0       0       0
       0       0       0       0       0       0       0       0       0       0
       0       0       0       0       0       0       0       0       0       0
       0       0       0       0       0       0       0       0       0
Stage Hydrograph TW Check=0
Use DSS=False
Use Fixed Start Time=False
Is Critical Boundary=False
Precipitation Mode=Disable
Wind Mode=No Wind Forces
Wave Mode=No Wave Forcing
Met BC=Precipitation|Expanded View=0
Met BC=Precipitation|Point Interpolation=Nearest
Met BC=Precipitation|Gridded Source=DSS
Met BC=Precipitation|Gridded Interpolation=
Met BC=Evapotranspiration|Expanded View=0
Met BC=Evapotranspiration|Point Interpolation=Nearest
Met BC=Evapotranspiration|Gridded Source=DSS
Met BC=Evapotranspiration|Gridded Interpolation=
Met BC=Wind Speed|Expanded View=0
Met BC=Wind Speed|Point Interpolation=Nearest
Met BC=Wind Speed|Gridded Source=DSS
Met BC=Wind Speed|Gridded Interpolation=
Met BC=Wind Direction|Expanded View=0
Met BC=Wind Direction|Point Interpolation=Nearest
Met BC=Wind Direction|Gridded Source=DSS
Met BC=Wind Direction|Gridded Interpolation=
Met BC=Wind Velocity X|Expanded View=0
Met BC=Wind Velocity X|Point Interpolation=Nearest
Met BC=Wind Velocity X|Gridded Source=DSS
Met BC=Wind Velocity X|Gridded Interpolation=
Met BC=Wind Velocity Y|Expanded View=0
Met BC=Wind Velocity Y|Point Interpolation=Nearest
Met BC=Wind Velocity Y|Gridded Source=DSS
Met BC=Wind Velocity Y|Gridded Interpolation=
Met BC=Wave Forcing X|Expanded View=0
Met BC=Wave Forcing X|Point Interpolation=Nearest
Met BC=Wave Forcing X|Gridded Source=DSS
Met BC=Wave Forcing X|Gridded Interpolation=
Met BC=Wave Forcing Y|Expanded View=0
Met BC=Wave Forcing Y|Point Interpolation=Nearest
Met BC=Wave Forcing Y|Gridded Source=DSS
Met BC=Wave Forcing Y|Gridded Interpolation=
Met BC=Air Density|Mode=Constant
Met BC=Air Density|Expanded View=0
Met BC=Air Density|Constant Value=1.225
Met BC=Air Density|Constant Units=kg/m3
Met BC=Air Density|Point Interpolation=Nearest
Met BC=Air Density|Gridded Source=DSS
Met BC=Air Density|Gridded Interpolation=
Met BC=Air Temperature|Expanded View=0
Met BC=Air Temperature|Point Interpolation=Nearest
Met BC=Air Temperature|Gridded Source=DSS
Met BC=Air Temperature|Gridded Interpolation=
Met BC=Humidity|Expanded View=0
Met BC=Humidity|Point Interpolation=Nearest
Met BC=Humidity|Gridded Source=DSS
Met BC=Humidity|Gridded Interpolation=
Met BC=Air Pressure|Mode=Constant
Met BC=Air Pressure|Expanded View=0
Met BC=Air Pressure|Constant Value=1013.2
Met BC=Air Pressure|Constant Units=mb
Met BC=Air Pressure|Point Interpolation=Inv Distance
Met BC=Air Pressure|Gridded Source=DSS
Met BC=Air Pressure|Gridded Interpolation=
Observed Time Series=Stage|TS Name=BC Line: DS Boundary
Observed Time Series=Stage|TS Used=-1
Observed Time Series=Stage|TS Source=DSS
Observed Time Series=Stage|TS DSS Filename=.\SWMM Extran Datasets\EXTRAN 1 example.dss
Observed Time Series=Stage|TS DSS Pathname=/Base/10208/Stage/01Jan1988/5Minute/EXTRAN 1 example/
Observed Time Series=Stage|TS Table Mode=0
Observed Time Series=Stage|TS Table Use Fixed Start=0
Observed Time Series=Stage|TS Table StartDateTime=01Jan1988 00:00:00
Observed Time Series=Stage|TS Table Interval=1 Hour
Observed Time Series=Stage|TS Table Data Units=ft
Observed Time Series=Stage|TS Table Data Type=INST-VAL
Observed Time Series=Stage|TS Constant Units=ft
Observed Time Series=Stage|TS Name=Pipe Node: Base [15009]
Observed Time Series=Stage|TS Used=-1
Observed Time Series=Stage|TS Source=DSS
Observed Time Series=Stage|TS DSS Filename=.\SWMM Extran Datasets\EXTRAN 1 example.dss
Observed Time Series=Stage|TS DSS Pathname=/Base/15009/Stage//5Minute/EXTRAN 1 example/
Observed Time Series=Stage|TS Table Mode=0
Observed Time Series=Stage|TS Table Use Fixed Start=0
Observed Time Series=Stage|TS Table StartDateTime=01Jan1988 00:00:00
Observed Time Series=Stage|TS Table Interval=1 Hour
Observed Time Series=Stage|TS Table Data Units=ft
Observed Time Series=Stage|TS Constant Units=ft
Observed Time Series=Stage|TS Name=Pipe Node: Base [81309]
Observed Time Series=Stage|TS Used=-1
Observed Time Series=Stage|TS Source=DSS
Observed Time Series=Stage|TS DSS Filename=.\SWMM Extran Datasets\EXTRAN 1 example.dss
Observed Time Series=Stage|TS DSS Pathname=/Base/81309/Stage//5Minute/EXTRAN 1 example/
Observed Time Series=Stage|TS Table Mode=0
Observed Time Series=Stage|TS Table Use Fixed Start=0
Observed Time Series=Stage|TS Table StartDateTime=01Jan1988 00:00:00
Observed Time Series=Stage|TS Table Interval=1 Hour
Observed Time Series=Stage|TS Name=Pipe Node: Base [81009]
Observed Time Series=Stage|TS Used=-1
Observed Time Series=Stage|TS Source=DSS
Observed Time Series=Stage|TS DSS Filename=.\SWMM Extran Datasets\EXTRAN 1 example.dss
Observed Time Series=Stage|TS DSS Pathname=/Base/81009/Stage//5Minute/EXTRAN 1 example/
Observed Time Series=Stage|TS Table Mode=0
Observed Time Series=Stage|TS Table Use Fixed Start=0
Observed Time Series=Stage|TS Table StartDateTime=01Jan1988 00:00:00
Observed Time Series=Stage|TS Table Interval=1 Hour
Observed Time Series=Stage|TS Name=Pipe Node: Base [16109]
Observed Time Series=Stage|TS Used=-1
Observed Time Series=Stage|TS Source=DSS
Observed Time Series=Stage|TS DSS Filename=.\SWMM Extran Datasets\EXTRAN 1 example.dss
Observed Time Series=Stage|TS DSS Pathname=/Base/16109/Stage//5Minute/EXTRAN 1 example/
Observed Time Series=Stage|TS Table Mode=0
Observed Time Series=Stage|TS Table Use Fixed Start=0
Observed Time Series=Stage|TS Table StartDateTime=01Jan1988 00:00:00
Observed Time Series=Stage|TS Table Interval=1 Hour
Observed Time Series=Stage|TS Table Data Units=ft
Observed Time Series=Stage|TS Table Data Type=INST-VAL
Observed Time Series=Stage|TS Constant Units=ft
Observed Time Series=Stage|TS Name=Pipe Node: Base [82309]
Observed Time Series=Stage|TS Used=-1
Observed Time Series=Stage|TS Source=DSS
Observed Time Series=Stage|TS DSS Filename=.\SWMM Extran Datasets\EXTRAN 1 example.dss
Observed Time Series=Stage|TS DSS Pathname=/Base/82309/Stage//5Minute/EXTRAN 1 example/
Observed Time Series=Stage|TS Table Mode=0
Observed Time Series=Stage|TS Table Use Fixed Start=0
Observed Time Series=Stage|TS Table StartDateTime=01Jan1988 00:00:00
Observed Time Series=Stage|TS Table Interval=1 Hour
Observed Time Series=Stage|TS Name=Pipe Node: Base [80608]
Observed Time Series=Stage|TS Used=-1
Observed Time Series=Stage|TS Source=DSS
Observed Time Series=Stage|TS DSS Filename=.\SWMM Extran Datasets\EXTRAN 1 example.dss
Observed Time Series=Stage|TS DSS Pathname=/Base/80608/Stage//5Minute/EXTRAN 1 example/
Observed Time Series=Stage|TS Table Mode=0
Observed Time Series=Stage|TS Table Use Fixed Start=0
Observed Time Series=Stage|TS Table StartDateTime=01Jan1988 00:00:00
Observed Time Series=Stage|TS Table Interval=1 Hour
Observed Time Series=Stage|TS Name=Pipe Node: Base [80408]
Observed Time Series=Stage|TS Used=-1
Observed Time Series=Stage|TS Source=DSS
Observed Time Series=Stage|TS DSS Filename=.\SWMM Extran Datasets\EXTRAN 1 example.dss
Observed Time Series=Stage|TS DSS Pathname=/Base/80408/Stage//5Minute/EXTRAN 1 example/
Observed Time Series=Stage|TS Table Mode=0
Observed Time Series=Stage|TS Table Use Fixed Start=0
Observed Time Series=Stage|TS Table StartDateTime=01Jan1988 00:00:00
Observed Time Series=Stage|TS Table Interval=1 Hour
Observed Time Series=Stage|TS Name=Pipe Node: Base [16009]
Observed Time Series=Stage|TS Used=-1
Observed Time Series=Stage|TS Source=DSS
Observed Time Series=Stage|TS DSS Filename=.\SWMM Extran Datasets\EXTRAN 1 example.dss
Observed Time Series=Stage|TS DSS Pathname=/Base/16009/Stage//5Minute/EXTRAN 1 example/
Observed Time Series=Stage|TS Table Mode=0
Observed Time Series=Stage|TS Table Use Fixed Start=0
Observed Time Series=Stage|TS Table Interval=1 Hour
Observed Time Series=Flow|TS Name=BC Line: DS Boundary
Observed Time Series=Flow|TS Used=-1
Observed Time Series=Flow|TS Source=DSS
Observed Time Series=Flow|TS DSS Filename=.\SWMM Extran Datasets\EXTRAN 1 example.dss
Observed Time Series=Flow|TS DSS Pathname=/Base/10208/Flow/01Jan1988/5Minute/EXTRAN 1 example/
Observed Time Series=Flow|TS Table Mode=0
Observed Time Series=Flow|TS Table Use Fixed Start=0
Observed Time Series=Flow|TS Table Interval=1 Hour
Observed Time Series=Flow|TS Table Data Units=cfs
Observed Time Series=Flow|TS Table Data Type=INST-VAL
Observed Time Series=Flow|TS Constant Units=cfs
Observed Time Series=Flow|TS Name=Pipe Node: Base [15009]
Observed Time Series=Flow|TS Used=-1
Observed Time Series=Flow|TS Source=DSS
Observed Time Series=Flow|TS DSS Filename=.\SWMM Extran Datasets\EXTRAN 1 example.dss
Observed Time Series=Flow|TS DSS Pathname=/Base/15009/Flow//5Minute/EXTRAN 1 example/
Observed Time Series=Flow|TS Table Mode=0
Observed Time Series=Flow|TS Table Use Fixed Start=0
Observed Time Series=Flow|TS Table StartDateTime=01Jan1988 00:00:00
Observed Time Series=Flow|TS Table Interval=1 Hour
Observed Time Series=Flow|TS Table Data Units=cfs
Observed Time Series=Flow|TS Constant Units=cfs
Observed Time Series=Flow|TS Name=Pipe Node: Base [81309]
Observed Time Series=Flow|TS Used=-1
Observed Time Series=Flow|TS Source=DSS
Observed Time Series=Flow|TS DSS Filename=.\SWMM Extran Datasets\EXTRAN 1 example.dss
Observed Time Series=Flow|TS DSS Pathname=/Base/81309/Flow//5Minute/EXTRAN 1 example/
Observed Time Series=Flow|TS Table Mode=0
Observed Time Series=Flow|TS Table Use Fixed Start=0
Observed Time Series=Flow|TS Table StartDateTime=01Jan1988 00:00:00
Observed Time Series=Flow|TS Table Interval=1 Hour
Observed Time Series=Flow|TS Table Data Units=cfs
Observed Time Series=Flow|TS Constant Units=cfs
Observed Time Series=Flow|TS Name=Pipe Node: Base [81009]
Observed Time Series=Flow|TS Used=-1
Observed Time Series=Flow|TS Source=DSS
Observed Time Series=Flow|TS DSS Filename=.\SWMM Extran Datasets\EXTRAN 1 example.dss
Observed Time Series=Flow|TS DSS Pathname=/Base/81009/Flow//5Minute/EXTRAN 1 example/
Observed Time Series=Flow|TS Table Mode=0
Observed Time Series=Flow|TS Table Use Fixed Start=0
Observed Time Series=Flow|TS Table StartDateTime=01Jan1988 00:00:00
Observed Time Series=Flow|TS Table Interval=1 Hour
Observed Time Series=Flow|TS Table Data Units=cfs
Observed Time Series=Flow|TS Constant Units=cfs
Observed Time Series=Flow|TS Name=Pipe Node: Base [16109]
Observed Time Series=Flow|TS Used=-1
Observed Time Series=Flow|TS Source=DSS
Observed Time Series=Flow|TS DSS Filename=.\SWMM Extran Datasets\EXTRAN 1 example.dss
Observed Time Series=Flow|TS DSS Pathname=/Base/16109/Flow//5Minute/EXTRAN 1 example/
Observed Time Series=Flow|TS Table Mode=0
Observed Time Series=Flow|TS Table Use Fixed Start=0
Observed Time Series=Flow|TS Table StartDateTime=01Jan1988 00:00:00
Observed Time Series=Flow|TS Table Interval=1 Hour
Observed Time Series=Flow|TS Table Data Units=cfs
Observed Time Series=Flow|TS Table Data Type=INST-VAL
Observed Time Series=Flow|TS Constant Units=cfs
Observed Time Series=Flow|TS Name=Pipe Node: Base [82309]
Observed Time Series=Flow|TS Used=-1
Observed Time Series=Flow|TS Source=DSS
Observed Time Series=Flow|TS DSS Filename=.\SWMM Extran Datasets\EXTRAN 1 example.dss
Observed Time Series=Flow|TS DSS Pathname=/Base/82309/Flow//5Minute/EXTRAN 1 example/
Observed Time Series=Flow|TS Table Mode=0
Observed Time Series=Flow|TS Table Use Fixed Start=0
Observed Time Series=Flow|TS Table StartDateTime=01Jan1988 00:00:00
Observed Time Series=Flow|TS Table Interval=1 Hour
Observed Time Series=Flow|TS Table Data Units=cfs
Observed Time Series=Flow|TS Constant Units=cfs
Observed Time Series=Flow|TS Name=Pipe Node: Base [80608]
Observed Time Series=Flow|TS Used=-1
Observed Time Series=Flow|TS Source=DSS
Observed Time Series=Flow|TS DSS Filename=.\SWMM Extran Datasets\EXTRAN 1 example.dss
Observed Time Series=Flow|TS DSS Pathname=/Base/80608/Flow//5Minute/EXTRAN 1 example/
Observed Time Series=Flow|TS Table Mode=0
Observed Time Series=Flow|TS Table Use Fixed Start=0
Observed Time Series=Flow|TS Table StartDateTime=01Jan1988 00:00:00
Observed Time Series=Flow|TS Table Interval=1 Hour
Observed Time Series=Flow|TS Table Data Units=cfs
Observed Time Series=Flow|TS Constant Units=cfs
Observed Time Series=Flow|TS Name=Pipe Node: Base [80408]
Observed Time Series=Flow|TS Used=-1
Observed Time Series=Flow|TS Source=DSS
Observed Time Series=Flow|TS DSS Filename=.\SWMM Extran Datasets\EXTRAN 1 example.dss
Observed Time Series=Flow|TS DSS Pathname=/Base/80408/Flow//5Minute/EXTRAN 1 example/
Observed Time Series=Flow|TS Table Mode=0
Observed Time Series=Flow|TS Table Use Fixed Start=0
Observed Time Series=Flow|TS Table StartDateTime=01Jan1988 00:00:00
Observed Time Series=Flow|TS Table Interval=1 Hour
Observed Time Series=Flow|TS Table Data Units=cfs
Observed Time Series=Flow|TS Constant Units=cfs
Observed Time Series=Flow|TS Name=Pipe Node: Base [16009]
Observed Time Series=Flow|TS Used=-1
Observed Time Series=Flow|TS Source=DSS
Observed Time Series=Flow|TS DSS Filename=.\SWMM Extran Datasets\EXTRAN 1 example.dss
Observed Time Series=Flow|TS DSS Pathname=/Base/16009/Flow//5Minute/EXTRAN 1 example/
Observed Time Series=Flow|TS Table Mode=0
Observed Time Series=Flow|TS Table Use Fixed Start=0
Observed Time Series=Flow|TS Table StartDateTime=01Jan1988 00:00:00
Observed Time Series=Flow|TS Table Interval=1 Hour
Observed Time Series=Flow|TS Table Data Units=cfs
Observed Time Series=Flow|TS Table Data Type=INST-VAL
Observed Time Series=Flow|TS Constant Units=cfs
Non-Newtonian Method= 0 ,
Non-Newtonian Constant Vol Conc=0
Non-Newtonian Yield Method= 0 ,
Non-Newtonian Yield Coef=0, 0
User Yeild=   0
Non-Newtonian Sed Visc= 0 ,
Non-Newtonian Obrian B=0
User Viscosity=0
User Viscosity Ratio=0
Herschel-Bulkley Coef=0, 0
Clastic Method= 0 ,
Coulomb Phi=0
Voellmy X=0
Non-Newtonian Hindered FV= 0
Non-Newtonian FV K=0
Non-Newtonian ds=0
Non-Newtonian Max Cv=0
Non-Newtonian Bulking Method= 0 ,
Non-Newtonian High C Transport= 0 ,
Lava Activation= 0
Temperature=1300,15,,15,14,980
Heat Ballance=1,1200,0.5,1,70,0.95
Viscosity=1000,,,
Profile Coefficient=4,1.3,
Lava Param=,2500,
