HEC-RAS study ExtranTestImport.prj: SWMM Extran Tests Circular

--- ExtranTestImport.u02 (unsteady flow) ---

Flow Title=Extran7 -InlinePump
Program Version=6.70
Use Restart= 0
Initial Storage Elev=Perimeter 1     ,94.4,0
Boundary Location=                ,                ,        ,        ,                ,Perimeter 1     ,                ,DS Boundary                     ,
Friction Slope=0.0035,0
Boundary Location=                ,                ,        ,        ,                ,                ,                ,                                ,Base [81009]
Interval=15MIN
Flow Hydrograph= 49
       0      50      50      50      50      50      50      50      50      50
      50      50      50       0       0       0       0       0       0       0
       0       0       0       0       0       0       0       0       0       0
       0       0       0       0       0       0       0       0       0       0
       0       0       0       0       0       0       0       0       0
Stage Hydrograph TW Check=0
Use DSS=False
Use Fixed Start Time=False
Is Critical Boundary=False
Boundary Location=                ,                ,        ,        ,                ,                ,                ,                                ,Base [82309]
Interval=15MIN
Flow Hydrograph= 49
       0      40      40      40      40      40      40      40      40      40
      40      40      40       0       0       0       0       0       0       0
       0       0       0       0       0       0       0       0       0       0
       0       0       0       0       0       0       0       0       0       0
       0       0       0       0       0       0       0       0       0
Stage Hydrograph TW Check=0
Use DSS=False
Use Fixed Start Time=False
Is Critical Boundary=False
Boundary Location=                ,                ,        ,        ,                ,                ,                ,                                ,Base [80408]
Interval=15MIN
Flow Hydrograph= 49
       0      45      45      45      45      45      45      45      45      45
      45      45      45       0       0       0       0       0       0       0
       0       0       0       0       0       0       0       0       0       0
       0       0       0       0       0       0       0       0       0       0
       0       0       0       0       0       0       0       0       0
Stage Hydrograph TW Check=0
Flow Hydrograph QMult= 0.5
Use DSS=False
Use Fixed Start Time=False
Is Critical Boundary=False
Boundary Location=                ,                ,        ,        ,                ,                ,Pump Station #1 ,                                ,
Rule Operation=Type=0,Var Type=1,Comment=Make a pump efficiency curve based on depth not head
Rule Operation=Type=1,Var Name=82309_Invert,Var Type=1,Real=112.2
Rule Operation=Type=2,Var Name=82309 WSEL,Var Type=1,PipeNode=Base [82309],Sim Group=Pipe Nodes,Sim Function=WS Elevation,Time=5,LBStart=0.16,LBEnd=0
Rule Operation=Type=0,Var Type=1,Comment=Compute the depth for the *cell*
Rule Operation=Type=5,Var Name=82309_Depth,Var Type=1,MathOperator1=2,MathOperator2=0,MathOperator3=0
Rule Expression=,Variable=82309 WSEL
Rule Expression=,Variable=82309_Invert
Rule Operation=Type=0,Var Type=1,Comment=Get the Pump Flow From the Table
Rule Operation=Type=6,Var Name=Table Pump Flow,Var Type=1,TableMode=3,Table2D=0,TableArgX=82309 Depth,TableArgY=
Rule Expression=,Variable=82309_Depth
Rule Table=6,1
       0       5     7.5      25    42.6    42.7
       0       5      10      20      20      20
Rule Operation=Type=0,Var Type=1,Comment=Set the pump flow from the table
Rule Operation=Type=3,Var Type=1,Sim Group=Pump Stations,Sim Function=Station.Pump Flow
Rule Expression=,Variable=Table Pump Flow
Precipitation Mode=Disable
Wind Mode=No Wind Forces
Wave Mode=No Wave Forcing
Met BC=Precipitation|Expanded View=0
Met BC=Precipitation|Point Interpolation=Nearest
Met BC=Precipitation|Gridded Source=DSS
Met BC=Precipitation|Gridded Interpolation=
Met BC=Evapotranspiration|Expanded View=0
Met BC=Evapotranspiration|Point Interpolation=Nearest
Met BC=Evapotranspiration|Gridded Source=DSS
Met BC=Evapotranspiration|Gridded Interpolation=
Met BC=Wind Speed|Expanded View=0
Met BC=Wind Speed|Point Interpolation=Nearest
Met BC=Wind Speed|Gridded Source=DSS
Met BC=Wind Speed|Gridded Interpolation=
Met BC=Wind Direction|Expanded View=0
Met BC=Wind Direction|Point Interpolation=Nearest
Met BC=Wind Direction|Gridded Source=DSS
Met BC=Wind Direction|Gridded Interpolation=
Met BC=Wind Velocity X|Expanded View=0
Met BC=Wind Velocity X|Point Interpolation=Nearest
Met BC=Wind Velocity X|Gridded Source=DSS
Met BC=Wind Velocity X|Gridded Interpolation=
Met BC=Wind Velocity Y|Expanded View=0
Met BC=Wind Velocity Y|Point Interpolation=Nearest
Met BC=Wind Velocity Y|Gridded Source=DSS
Met BC=Wind Velocity Y|Gridded Interpolation=
Met BC=Wave Forcing X|Expanded View=0
Met BC=Wave Forcing X|Point Interpolation=Nearest
Met BC=Wave Forcing X|Gridded Source=DSS
Met BC=Wave Forcing X|Gridded Interpolation=
Met BC=Wave Forcing Y|Expanded View=0
Met BC=Wave Forcing Y|Point Interpolation=Nearest
Met BC=Wave Forcing Y|Gridded Source=DSS
Met BC=Wave Forcing Y|Gridded Interpolation=
Met BC=Air Density|Mode=Constant
Met BC=Air Density|Expanded View=0
Met BC=Air Density|Constant Value=1.225
Met BC=Air Density|Constant Units=kg/m3
Met BC=Air Density|Point Interpolation=Nearest
Met BC=Air Density|Gridded Source=DSS
Met BC=Air Density|Gridded Interpolation=
Met BC=Air Temperature|Expanded View=0
Met BC=Air Temperature|Point Interpolation=Nearest
Met BC=Air Temperature|Gridded Source=DSS
Met BC=Air Temperature|Gridded Interpolation=
Met BC=Humidity|Expanded View=0
Met BC=Humidity|Point Interpolation=Nearest
Met BC=Humidity|Gridded Source=DSS
Met BC=Humidity|Gridded Interpolation=
Met BC=Air Pressure|Mode=Constant
Met BC=Air Pressure|Expanded View=0
Met BC=Air Pressure|Constant Value=1013.2
Met BC=Air Pressure|Constant Units=mb
Met BC=Air Pressure|Point Interpolation=
Met BC=Air Pressure|Gridded Source=DSS
Met BC=Air Pressure|Gridded Interpolation=
Observed Time Series=Stage|TS Name=BC Line: DS Boundary
Observed Time Series=Stage|TS Used=-1
Observed Time Series=Stage|TS Source=DSS
Observed Time Series=Stage|TS DSS Filename=.\SWMM Extran Datasets\EXTRAN 7 Example.dss
Observed Time Series=Stage|TS DSS Pathname=/Base/10208/Flow/01Jan1988/5Minute/EXTRAN 6 Example/
Observed Time Series=Stage|TS Table Mode=0
Observed Time Series=Stage|TS Table Use Fixed Start=0
Observed Time Series=Stage|TS Table Interval=1 Hour
Observed Time Series=Stage|TS Table Data Units=ft
Observed Time Series=Stage|TS Table Data Type=INST-VAL
Observed Time Series=Stage|TS Constant Units=ft
Observed Time Series=Stage|TS Name=Pipe Node: Base [15009]
Observed Time Series=Stage|TS Used=-1
Observed Time Series=Stage|TS Source=DSS
Observed Time Series=Stage|TS DSS Filename=.\SWMM Extran Datasets\EXTRAN 7 Example.dss
Observed Time Series=Stage|TS DSS Pathname=/Base/15009/Stage//5Minute/EXTRAN 6 example/
Observed Time Series=Stage|TS Table Mode=0
Observed Time Series=Stage|TS Table Use Fixed Start=0
Observed Time Series=Stage|TS Table Interval=1 Hour
Observed Time Series=Stage|TS Name=Pipe Node: Base [81309]
Observed Time Series=Stage|TS Used=-1
Observed Time Series=Stage|TS Source=DSS
Observed Time Series=Stage|TS DSS Filename=.\SWMM Extran Datasets\EXTRAN 7 Example.dss
Observed Time Series=Stage|TS DSS Pathname=/Base/81309/Stage//5Minute/EXTRAN 6 example/
Observed Time Series=Stage|TS Table Mode=0
Observed Time Series=Stage|TS Table Use Fixed Start=0
Observed Time Series=Stage|TS Table Interval=1 Hour
Observed Time Series=Stage|TS Name=Pipe Node: Base [81009]
Observed Time Series=Stage|TS Used=-1
Observed Time Series=Stage|TS Source=DSS
Observed Time Series=Stage|TS DSS Filename=.\SWMM Extran Datasets\EXTRAN 7 Example.dss
Observed Time Series=Stage|TS DSS Pathname=/Base/81009/Stage//5Minute/EXTRAN 6 example/
Observed Time Series=Stage|TS Table Mode=0
Observed Time Series=Stage|TS Table Use Fixed Start=0
Observed Time Series=Stage|TS Table Interval=1 Hour
Observed Time Series=Stage|TS Name=Pipe Node: Base [16109]
Observed Time Series=Stage|TS Used=-1
Observed Time Series=Stage|TS Source=DSS
Observed Time Series=Stage|TS DSS Filename=.\SWMM Extran Datasets\EXTRAN 7 Example.dss
Observed Time Series=Stage|TS DSS Pathname=/Base/16109/Stage//5Minute/EXTRAN 6 example/
Observed Time Series=Stage|TS Table Mode=0
Observed Time Series=Stage|TS Table Use Fixed Start=0
Observed Time Series=Stage|TS Table StartDateTime=01Jan1988 00:00:00
Observed Time Series=Stage|TS Table Interval=1 Hour
Observed Time Series=Stage|TS Table Data Units=ft
Observed Time Series=Stage|TS Table Data Type=INST-VAL
Observed Time Series=Stage|TS Constant Units=ft
Observed Time Series=Stage|TS Name=Pipe Node: Base [82309]
Observed Time Series=Stage|TS Used=-1
Observed Time Series=Stage|TS Source=DSS
Observed Time Series=Stage|TS DSS Filename=.\SWMM Extran Datasets\EXTRAN 7 Example.dss
Observed Time Series=Stage|TS DSS Pathname=/Base/82309/Stage//5Minute/EXTRAN 6 example/
Observed Time Series=Stage|TS Table Mode=0
Observed Time Series=Stage|TS Table Use Fixed Start=0
Observed Time Series=Stage|TS Table Interval=1 Hour
Observed Time Series=Stage|TS Name=Pipe Node: Base [80608]
Observed Time Series=Stage|TS Used=-1
Observed Time Series=Stage|TS Source=DSS
Observed Time Series=Stage|TS DSS Filename=.\SWMM Extran Datasets\EXTRAN 7 Example.dss
Observed Time Series=Stage|TS DSS Pathname=/Base/80608/Stage//5Minute/EXTRAN 6 example/
Observed Time Series=Stage|TS Table Mode=0
Observed Time Series=Stage|TS Table Use Fixed Start=0
Observed Time Series=Stage|TS Table Interval=1 Hour
Observed Time Series=Stage|TS Name=Pipe Node: Base [80408]
Observed Time Series=Stage|TS Used=-1
Observed Time Series=Stage|TS Source=DSS
Observed Time Series=Stage|TS DSS Filename=.\SWMM Extran Datasets\EXTRAN 7 Example.dss
Observed Time Series=Stage|TS DSS Pathname=/Base/80408/Stage//5Minute/EXTRAN 6 example/
Observed Time Series=Stage|TS Table Mode=0
Observed Time Series=Stage|TS Table Use Fixed Start=0
Observed Time Series=Stage|TS Table Interval=1 Hour
Observed Time Series=Stage|TS Name=Pipe Node: Base [16009]
Observed Time Series=Stage|TS Used=-1
Observed Time Series=Stage|TS Source=DSS
Observed Time Series=Stage|TS DSS Filename=.\SWMM Extran Datasets\EXTRAN 7 Example.dss
Observed Time Series=Stage|TS DSS Pathname=/Base/16009/Stage//5Minute/EXTRAN 6 example/
Observed Time Series=Stage|TS Table Mode=0
Observed Time Series=Stage|TS Table Use Fixed Start=0
Observed Time Series=Stage|TS Table Interval=1 Hour
Observed Time Series=Flow|TS Name=BC Line: DS Boundary
Observed Time Series=Flow|TS Used=-1
Observed Time Series=Flow|TS Source=DSS
Observed Time Series=Flow|TS DSS Filename=.\SWMM Extran Datasets\EXTRAN 7 Example.dss
Observed Time Series=Flow|TS DSS Pathname=/Base/10208/Flow/01Jan1988/5Minute/EXTRAN 6 example/
Observed Time Series=Flow|TS Table Mode=0
Observed Time Series=Flow|TS Table Use Fixed Start=0
Observed Time Series=Flow|TS Table StartDateTime=01Jan1988 00:00:00
Observed Time Series=Flow|TS Table Interval=1 Hour
Observed Time Series=Flow|TS Table Data Units=cfs
Observed Time Series=Flow|TS Table Data Type=INST-VAL
Observed Time Series=Flow|TS Constant Units=cfs
Observed Time Series=Flow|TS Name=Pipe Node: Base [15009]
Observed Time Series=Flow|TS Used=-1
Observed Time Series=Flow|TS Source=DSS
Observed Time Series=Flow|TS DSS Filename=.\SWMM Extran Datasets\EXTRAN 7 Example.dss
Observed Time Series=Flow|TS DSS Pathname=/Base/15009/Flow//5Minute/EXTRAN 6 example/
Observed Time Series=Flow|TS Table Mode=0
Observed Time Series=Flow|TS Table Use Fixed Start=0
Observed Time Series=Flow|TS Table StartDateTime=01Jan1988 00:00:00
Observed Time Series=Flow|TS Table Interval=1 Hour
Observed Time Series=Flow|TS Table Data Units=cfs
Observed Time Series=Flow|TS Constant Units=cfs
Observed Time Series=Flow|TS Name=Pipe Node: Base [81309]
Observed Time Series=Flow|TS Used=-1
Observed Time Series=Flow|TS Source=DSS
Observed Time Series=Flow|TS DSS Filename=.\SWMM Extran Datasets\EXTRAN 7 Example.dss
Observed Time Series=Flow|TS DSS Pathname=/Base/81309/Flow//5Minute/EXTRAN 6 example/
Observed Time Series=Flow|TS Table Mode=0
Observed Time Series=Flow|TS Table Use Fixed Start=0
Observed Time Series=Flow|TS Table StartDateTime=01Jan1988 00:00:00
Observed Time Series=Flow|TS Table Interval=1 Hour
Observed Time Series=Flow|TS Table Data Units=cfs
Observed Time Series=Flow|TS Constant Units=cfs
Observed Time Series=Flow|TS Name=Pipe Node: Base [81009]
Observed Time Series=Flow|TS Used=-1
Observed Time Series=Flow|TS Source=DSS
Observed Time Series=Flow|TS DSS Filename=.\SWMM Extran Datasets\EXTRAN 7 Example.dss
Observed Time Series=Flow|TS DSS Pathname=/Base/81009/Flow//5Minute/EXTRAN 6 example/
Observed Time Series=Flow|TS Table Mode=0
Observed Time Series=Flow|TS Table Use Fixed Start=0
Observed Time Series=Flow|TS Table StartDateTime=01Jan1988 00:00:00
Observed Time Series=Flow|TS Table Interval=1 Hour
Observed Time Series=Flow|TS Table Data Units=cfs
Observed Time Series=Flow|TS Constant Units=cfs
Observed Time Series=Flow|TS Name=Pipe Node: Base [16109]
Observed Time Series=Flow|TS Used=-1
Observed Time Series=Flow|TS Source=DSS
Observed Time Series=Flow|TS DSS Filename=.\SWMM Extran Datasets\EXTRAN 7 Example.dss
Observed Time Series=Flow|TS DSS Pathname=/Base/16109/Flow//5Minute/EXTRAN 6 example/
Observed Time Series=Flow|TS Table Mode=0
Observed Time Series=Flow|TS Table Use Fixed Start=0
Observed Time Series=Flow|TS Table StartDateTime=01Jan1988 00:00:00
Observed Time Series=Flow|TS Table Interval=1 Hour
Observed Time Series=Flow|TS Table Data Units=cfs
Observed Time Series=Flow|TS Table Data Type=INST-VAL
Observed Time Series=Flow|TS Constant Units=cfs
Observed Time Series=Flow|TS Name=Pipe Node: Base [82309]
Observed Time Series=Flow|TS Used=-1
Observed Time Series=Flow|TS Source=DSS
Observed Time Series=Flow|TS DSS Filename=.\SWMM Extran Datasets\EXTRAN 7 Example.dss
Observed Time Series=Flow|TS DSS Pathname=/Base/82309/Flow//5Minute/EXTRAN 6 example/
Observed Time Series=Flow|TS Table Mode=0
Observed Time Series=Flow|TS Table Use Fixed Start=0
Observed Time Series=Flow|TS Table StartDateTime=01Jan1988 00:00:00
Observed Time Series=Flow|TS Table Interval=1 Hour
Observed Time Series=Flow|TS Table Data Units=cfs
Observed Time Series=Flow|TS Constant Units=cfs
Observed Time Series=Flow|TS Name=Pipe Node: Base [80608]
Observed Time Series=Flow|TS Used=-1
Observed Time Series=Flow|TS Source=DSS
Observed Time Series=Flow|TS DSS Filename=.\SWMM Extran Datasets\EXTRAN 7 Example.dss
Observed Time Series=Flow|TS DSS Pathname=/Base/80608/Flow//5Minute/EXTRAN 6 example/
Observed Time Series=Flow|TS Table Mode=0
Observed Time Series=Flow|TS Table Use Fixed Start=0
Observed Time Series=Flow|TS Table StartDateTime=01Jan1988 00:00:00
Observed Time Series=Flow|TS Table Interval=1 Hour
Observed Time Series=Flow|TS Table Data Units=cfs
Observed Time Series=Flow|TS Constant Units=cfs
Observed Time Series=Flow|TS Name=Pipe Node: Base [80408]
Observed Time Series=Flow|TS Used=-1
Observed Time Series=Flow|TS Source=DSS
Observed Time Series=Flow|TS DSS Filename=.\SWMM Extran Datasets\EXTRAN 7 Example.dss
Observed Time Series=Flow|TS DSS Pathname=/Base/80408/Flow//5Minute/EXTRAN 6 example/
Observed Time Series=Flow|TS Table Mode=0
Observed Time Series=Flow|TS Table Use Fixed Start=0
Observed Time Series=Flow|TS Table StartDateTime=01Jan1988 00:00:00
Observed Time Series=Flow|TS Table Interval=1 Hour
Observed Time Series=Flow|TS Table Data Units=cfs
Observed Time Series=Flow|TS Constant Units=cfs
Observed Time Series=Flow|TS Name=Pipe Node: Base [16009]
Observed Time Series=Flow|TS Used=-1
Observed Time Series=Flow|TS Source=DSS
Observed Time Series=Flow|TS DSS Filename=.\SWMM Extran Datasets\EXTRAN 7 Example.dss
Observed Time Series=Flow|TS DSS Pathname=/Base/16009/Flow//5Minute/EXTRAN 6 example/
Observed Time Series=Flow|TS Table Mode=0
Observed Time Series=Flow|TS Table Use Fixed Start=0
Observed Time Series=Flow|TS Table StartDateTime=01Jan1988 00:00:00
Observed Time Series=Flow|TS Table Interval=1 Hour
Observed Time Series=Flow|TS Table Data Units=cfs
Observed Time Series=Flow|TS Table Data Type=INST-VAL
Observed Time Series=Flow|TS Constant Units=cfs
Non-Newtonian Method= 0 ,
Non-Newtonian Constant Vol Conc=0
Non-Newtonian Yield Method= 0 ,
Non-Newtonian Yield Coef=0, 0
User Yeild=   0
Non-Newtonian Sed Visc= 0 ,
Non-Newtonian Obrian B=0
User Viscosity=0
User Viscosity Ratio=0
Herschel-Bulkley Coef=0, 0
Clastic Method= 0 ,
Coulomb Phi=0
Voellmy X=0
Non-Newtonian Hindered FV= 0
Non-Newtonian FV K=0
Non-Newtonian ds=0
Non-Newtonian Max Cv=0
Non-Newtonian Bulking Method= 0 ,
Non-Newtonian High C Transport= 0 ,
Lava Activation= 0
Temperature=1300,15,,15,14,980
Heat Ballance=1,1200,0.5,1,70,0.95
Viscosity=1000,,,
Profile Coefficient=4,1.3,
Lava Param=,2500,

--- ExtranTestImport.u04 (unsteady flow) ---

Flow Title=Extran2
Program Version=7.00
Use Restart= 0
Boundary Location=                ,                ,        ,        ,                ,Perimeter 1     ,                ,DS Boundary                     ,                                ,
Interval=1DAY
Stage Hydrograph= 2
    94.4    94.4
Stage Hydrograph Use Initial Stage=-1
Stage Hydrograph TW Check=0
Use DSS=False
Use Fixed Start Time=False
Is Critical Boundary=False
Boundary Location=                ,                ,        ,        ,                ,                ,                ,                                ,Base [81009]                    ,
Interval=15MIN
Flow Hydrograph= 49
       0      50      50      50      50      50      50      50      50      50
      50      50      50       0       0       0       0       0       0       0
       0       0       0       0       0       0       0       0       0       0
       0       0       0       0       0       0       0       0       0       0
       0       0       0       0       0       0       0       0       0
Stage Hydrograph TW Check=0
Use DSS=False
Use Fixed Start Time=False
Is Critical Boundary=False
Boundary Location=                ,                ,        ,        ,                ,                ,                ,                                ,Base [82309]                    ,
Interval=15MIN
Flow Hydrograph= 49
       0      40      40      40      40      40      40      40      40      40
      40      40      40       0       0       0       0       0       0       0
       0       0       0       0       0       0       0       0       0       0
       0       0       0       0       0       0       0       0       0       0
       0       0       0       0       0       0       0       0       0
Stage Hydrograph TW Check=0
Use DSS=False
Use Fixed Start Time=False
Is Critical Boundary=False
Boundary Location=                ,                ,        ,        ,                ,                ,                ,                                ,Base [80408]                    ,
Interval=15MIN
Flow Hydrograph= 49
       0      45      45      45      45      45      45      45      45      45
      45      45      45       0       0       0       0       0       0       0
       0       0       0       0       0       0       0       0       0       0
       0       0       0       0       0       0       0       0       0       0
       0       0       0       0       0       0       0       0       0
Stage Hydrograph TW Check=0
Use DSS=False
Use Fixed Start Time=False
Is Critical Boundary=False
Precipitation Mode=Disable
Wind Mode=No Wind Forces
Wave Mode=No Wave Forcing
Met BC=Precipitation|Expanded View=0
Met BC=Precipitation|Point Interpolation=Nearest
Met BC=Precipitation|Gridded Source=DSS
Met BC=Precipitation|Gridded Interpolation=
Met BC=Evapotranspiration|Expanded View=0
Met BC=Evapotranspiration|Point Interpolation=Nearest
Met BC=Evapotranspiration|Gridded Source=DSS
Met BC=Evapotranspiration|Gridded Interpolation=
Met BC=Wind Speed|Expanded View=0
Met BC=Wind Speed|Point Interpolation=Nearest
Met BC=Wind Speed|Gridded Source=DSS
Met BC=Wind Speed|Gridded Interpolation=
Met BC=Wind Direction|Expanded View=0
Met BC=Wind Direction|Point Interpolation=Nearest
Met BC=Wind Direction|Gridded Source=DSS
Met BC=Wind Direction|Gridded Interpolation=
Met BC=Wind Velocity X|Expanded View=0
Met BC=Wind Velocity X|Point Interpolation=Nearest
Met BC=Wind Velocity X|Gridded Source=DSS
Met BC=Wind Velocity X|Gridded Interpolation=
Met BC=Wind Velocity Y|Expanded View=0
Met BC=Wind Velocity Y|Point Interpolation=Nearest
Met BC=Wind Velocity Y|Gridded Source=DSS
Met BC=Wind Velocity Y|Gridded Interpolation=
Met BC=Wave Forcing X|Expanded View=0
Met BC=Wave Forcing X|Point Interpolation=Nearest
Met BC=Wave Forcing X|Gridded Source=DSS
Met BC=Wave Forcing X|Gridded Interpolation=
Met BC=Wave Forcing Y|Expanded View=0
Met BC=Wave Forcing Y|Point Interpolation=Nearest
Met BC=Wave Forcing Y|Gridded Source=DSS
Met BC=Wave Forcing Y|Gridded Interpolation=
Met BC=Air Density|Mode=Constant
Met BC=Air Density|Expanded View=0
Met BC=Air Density|Constant Value=1.225
Met BC=Air Density|Constant Units=kg/m3
Met BC=Air Density|Point Interpolation=Nearest
Met BC=Air Density|Gridded Source=DSS
Met BC=Air Density|Gridded Interpolation=
Met BC=Air Temperature|Expanded View=0
Met BC=Air Temperature|Point Interpolation=Nearest
Met BC=Air Temperature|Gridded Source=DSS
Met BC=Air Temperature|Gridded Interpolation=
Met BC=Humidity|Expanded View=0
Met BC=Humidity|Point Interpolation=Nearest
Met BC=Humidity|Gridded Source=DSS
Met BC=Humidity|Gridded Interpolation=
Met BC=Air Pressure|Mode=Constant
Met BC=Air Pressure|Expanded View=0
Met BC=Air Pressure|Constant Value=1013.2
Met BC=Air Pressure|Constant Units=mb
Met BC=Air Pressure|Point Interpolation=
Met BC=Air Pressure|Gridded Source=DSS
Met BC=Air Pressure|Gridded Interpolation=
Observed Time Series=Stage|TS Name=Pipe Node: Base [15009]
Observed Time Series=Stage|TS Used=-1
Observed Time Series=Stage|TS Source=DSS
Observed Time Series=Stage|TS DSS Filename=.\SWMM Extran Datasets\EXTRAN 2 example.dss
Observed Time Series=Stage|TS DSS Pathname=/Base/15009/Stage//5Minute/EXTRAN 2 example/
Observed Time Series=Stage|TS Table Mode=0
Observed Time Series=Stage|TS Table Use Fixed Start=0
Observed Time Series=Stage|TS Table Interval=1 Hour
Observed Time Series=Stage|TS Name=Pipe Node: Base [16009]
Observed Time Series=Stage|TS Used=-1
Observed Time Series=Stage|TS Source=DSS
Observed Time Series=Stage|TS DSS Filename=.\SWMM Extran Datasets\EXTRAN 2 example.dss
Observed Time Series=Stage|TS DSS Pathname=/Base/16009/Stage//5Minute/EXTRAN 2 example/
Observed Time Series=Stage|TS Table Mode=0
Observed Time Series=Stage|TS Table Use Fixed Start=0
Observed Time Series=Stage|TS Table Interval=1 Hour
Observed Time Series=Stage|TS Name=Pipe Node: Base [16109]
Observed Time Series=Stage|TS Used=-1
Observed Time Series=Stage|TS Source=DSS
Observed Time Series=Stage|TS DSS Filename=.\SWMM Extran Datasets\EXTRAN 2 example.dss
Observed Time Series=Stage|TS DSS Pathname=/Base/16109/Stage//5Minute/EXTRAN 2 example/
Observed Time Series=Stage|TS Table Mode=0
Observed Time Series=Stage|TS Table Use Fixed Start=0
Observed Time Series=Stage|TS Table Interval=1 Hour
Observed Time Series=Stage|TS Name=Pipe Node: Base [80408]
Observed Time Series=Stage|TS Used=-1
Observed Time Series=Stage|TS Source=DSS
Observed Time Series=Stage|TS DSS Filename=.\SWMM Extran Datasets\EXTRAN 2 example.dss
Observed Time Series=Stage|TS DSS Pathname=/Base/80408/Stage//5Minute/EXTRAN 2 example/
Observed Time Series=Stage|TS Table Mode=0
Observed Time Series=Stage|TS Table Use Fixed Start=0
Observed Time Series=Stage|TS Table Interval=1 Hour
Observed Time Series=Stage|TS Name=Pipe Node: Base [80608]
Observed Time Series=Stage|TS Used=-1
Observed Time Series=Stage|TS Source=DSS
Observed Time Series=Stage|TS DSS Filename=.\SWMM Extran Datasets\EXTRAN 2 example.dss
Observed Time Series=Stage|TS DSS Pathname=/Base/80608/Stage//5Minute/EXTRAN 2 example/
Observed Time Series=Stage|TS Table Mode=0
Observed Time Series=Stage|TS Table Use Fixed Start=0
Observed Time Series=Stage|TS Table Interval=1 Hour
Observed Time Series=Stage|TS Name=Pipe Node: Base [81009]
Observed Time Series=Stage|TS Used=-1
Observed Time Series=Stage|TS Source=DSS
Observed Time Series=Stage|TS DSS Filename=.\SWMM Extran Datasets\EXTRAN 2 example.dss
Observed Time Series=Stage|TS DSS Pathname=/Base/81009/Stage//5Minute/EXTRAN 2 example/
Observed Time Series=Stage|TS Table Mode=0
Observed Time Series=Stage|TS Table Use Fixed Start=0
Observed Time Series=Stage|TS Table Interval=1 Hour
Observed Time Series=Stage|TS Name=Pipe Node: Base [81309]
Observed Time Series=Stage|TS Used=-1
Observed Time Series=Stage|TS Source=DSS
Observed Time Series=Stage|TS DSS Filename=.\SWMM Extran Datasets\EXTRAN 2 example.dss
Observed Time Series=Stage|TS DSS Pathname=/Base/81309/Stage//5Minute/EXTRAN 2 example/
Observed Time Series=Stage|TS Table Mode=0
Observed Time Series=Stage|TS Table Use Fixed Start=0
Observed Time Series=Stage|TS Table Interval=1 Hour
Observed Time Series=Stage|TS Name=Pipe Node: Base [82309]
Observed Time Series=Stage|TS Used=-1
Observed Time Series=Stage|TS Source=DSS
Observed Time Series=Stage|TS DSS Filename=.\SWMM Extran Datasets\EXTRAN 2 example.dss
Observed Time Series=Stage|TS DSS Pathname=/Base/82309/Stage//5Minute/EXTRAN 2 example/
Observed Time Series=Stage|TS Table Mode=0
Observed Time Series=Stage|TS Table Use Fixed Start=0
Observed Time Series=Stage|TS Table Interval=1 Hour
Observed Time Series=Flow|TS Name=Pipe Node: Base [15009]
Observed Time Series=Flow|TS Used=-1
Observed Time Series=Flow|TS Source=DSS
Observed Time Series=Flow|TS DSS Filename=.\SWMM Extran Datasets\EXTRAN 2 example.dss
Observed Time Series=Flow|TS DSS Pathname=/Base/15009/Flow//5Minute/EXTRAN 2 example/
Observed Time Series=Flow|TS Table Mode=0
Observed Time Series=Flow|TS Table Use Fixed Start=0
Observed Time Series=Flow|TS Table Interval=1 Hour
Observed Time Series=Flow|TS Name=Pipe Node: Base [16009]
Observed Time Series=Flow|TS Used=-1
Observed Time Series=Flow|TS Source=DSS
Observed Time Series=Flow|TS DSS Filename=.\SWMM Extran Datasets\EXTRAN 2 example.dss
Observed Time Series=Flow|TS DSS Pathname=/Base/16009/Flow//5Minute/EXTRAN 2 example/
Observed Time Series=Flow|TS Table Mode=0
Observed Time Series=Flow|TS Table Use Fixed Start=0
Observed Time Series=Flow|TS Table Interval=1 Hour
Observed Time Series=Flow|TS Name=Pipe Node: Base [16109]
Observed Time Series=Flow|TS Used=-1
Observed Time Series=Flow|TS Source=DSS
Observed Time Series=Flow|TS DSS Filename=.\SWMM Extran Datasets\EXTRAN 2 example.dss
Observed Time Series=Flow|TS DSS Pathname=/Base/16109/Flow//5Minute/EXTRAN 2 example/
Observed Time Series=Flow|TS Table Mode=0
Observed Time Series=Flow|TS Table Use Fixed Start=0
Observed Time Series=Flow|TS Table Interval=1 Hour
Observed Time Series=Flow|TS Name=Pipe Node: Base [80408]
Observed Time Series=Flow|TS Used=-1
Observed Time Series=Flow|TS Source=DSS
Observed Time Series=Flow|TS DSS Filename=.\SWMM Extran Datasets\EXTRAN 2 example.dss
Observed Time Series=Flow|TS DSS Pathname=/Base/80408/Flow//5Minute/EXTRAN 2 example/
Observed Time Series=Flow|TS Table Mode=0
Observed Time Series=Flow|TS Table Use Fixed Start=0
Observed Time Series=Flow|TS Table Interval=1 Hour
Observed Time Series=Flow|TS Name=Pipe Node: Base [80608]
Observed Time Series=Flow|TS Used=-1
Observed Time Series=Flow|TS Source=DSS
Observed Time Series=Flow|TS DSS Filename=.\SWMM Extran Datasets\EXTRAN 2 example.dss
Observed Time Series=Flow|TS DSS Pathname=/Base/80608/Flow//5Minute/EXTRAN 2 example/
Observed Time Series=Flow|TS Table Mode=0
Observed Time Series=Flow|TS Table Use Fixed Start=0
Observed Time Series=Flow|TS Table Interval=1 Hour
Observed Time Series=Flow|TS Name=Pipe Node: Base [81009]
Observed Time Series=Flow|TS Used=-1
Observed Time Series=Flow|TS Source=DSS
Observed Time Series=Flow|TS DSS Filename=.\SWMM Extran Datasets\EXTRAN 2 example.dss
Observed Time Series=Flow|TS DSS Pathname=/Base/81009/Flow//5Minute/EXTRAN 2 example/
Observed Time Series=Flow|TS Table Mode=0
Observed Time Series=Flow|TS Table Use Fixed Start=0
Observed Time Series=Flow|TS Table Interval=1 Hour
Observed Time Series=Flow|TS Name=Pipe Node: Base [81309]
Observed Time Series=Flow|TS Used=-1
Observed Time Series=Flow|TS Source=DSS
Observed Time Series=Flow|TS DSS Filename=.\SWMM Extran Datasets\EXTRAN 2 example.dss
Observed Time Series=Flow|TS DSS Pathname=/Base/81309/Flow//5Minute/EXTRAN 2 example/
Observed Time Series=Flow|TS Table Mode=0
Observed Time Series=Flow|TS Table Use Fixed Start=0
Observed Time Series=Flow|TS Table Interval=1 Hour
Observed Time Series=Flow|TS Name=Pipe Node: Base [82309]
Observed Time Series=Flow|TS Used=-1
Observed Time Series=Flow|TS Source=DSS
Observed Time Series=Flow|TS DSS Filename=.\SWMM Extran Datasets\EXTRAN 2 example.dss
Observed Time Series=Flow|TS DSS Pathname=/Base/82309/Flow//5Minute/EXTRAN 2 example/
Observed Time Series=Flow|TS Table Mode=0
Observed Time Series=Flow|TS Table Use Fixed Start=0
Observed Time Series=Flow|TS Table Interval=1 Hour
Non-Newtonian Method= 0 ,
Non-Newtonian Constant Vol Conc=0
Non-Newtonian Yield Method= 0 ,
Non-Newtonian Yield Coef=0, 0
User Yeild=   0
Non-Newtonian Sed Visc= 0 ,
Non-Newtonian Obrian B=0
User Viscosity=0
User Viscosity Ratio=0
Herschel-Bulkley Coef=0, 0
Clastic Method= 0 ,
Coulomb Phi=0
Voellmy X=0
Non-Newtonian Hindered FV= 0
Non-Newtonian FV K=0
Non-Newtonian ds=0
Non-Newtonian Max Cv=0
Non-Newtonian Bulking Method= 0 ,
Non-Newtonian High C Transport= 0 ,
Lava Activation= 0
Temperature=1300,15,,15,14,980
Heat Ballance=1,1200,0.5,1,70,0.95
Viscosity=1000,,,
Profile Coefficient=4,1.3,
Lava Param=,2500,

--- ExtranTestImport.u06 (unsteady flow) ---

Flow Title=Extran 4
Program Version=7.00
Use Restart= 0
Boundary Location=                ,                ,        ,        ,                ,Perimeter 1     ,                ,DS Boundary                     ,                                ,
Friction Slope=0.0045
Boundary Location=                ,                ,        ,        ,                ,                ,                ,                                ,Base [81009]                    ,
Interval=15MIN
Flow Hydrograph= 49
       0      50      50      50      50      50      50      50      50      50
      50      50      50       0       0       0       0       0       0       0
       0       0       0       0       0       0       0       0       0       0
       0       0       0       0       0       0       0       0       0       0
       0       0       0       0       0       0       0       0       0
Stage Hydrograph TW Check=0
Use DSS=False
Use Fixed Start Time=False
Is Critical Boundary=False
Boundary Location=                ,                ,        ,        ,                ,                ,                ,                                ,Base [82309]                    ,
Interval=15MIN
Flow Hydrograph= 49
       0      40      40      40      40      40      40      40      40      40
      40      40      40       0       0       0       0       0       0       0
       0       0       0       0       0       0       0       0       0       0
       0       0       0       0       0       0       0       0       0       0
       0       0       0       0       0       0       0       0       0
Stage Hydrograph TW Check=0
Use DSS=False
Use Fixed Start Time=False
Is Critical Boundary=False
Boundary Location=                ,                ,        ,        ,                ,                ,                ,                                ,Base [80408]                    ,
Interval=15MIN
Flow Hydrograph= 49
       0      45      45      45      45      45      45      45      45      45
      45      45      45       0       0       0       0       0       0       0
       0       0       0       0       0       0       0       0       0       0
       0       0       0       0       0       0       0       0       0       0
       0       0       0       0       0       0       0       0       0
Stage Hydrograph TW Check=0
Use DSS=False
Use Fixed Start Time=False
Is Critical Boundary=False
Precipitation Mode=Disable
Wind Mode=No Wind Forces
Wave Mode=No Wave Forcing
Met BC=Precipitation|Expanded View=0
Met BC=Precipitation|Point Interpolation=Nearest
Met BC=Precipitation|Gridded Source=DSS
Met BC=Precipitation|Gridded Interpolation=
Met BC=Evapotranspiration|Expanded View=0
Met BC=Evapotranspiration|Point Interpolation=Nearest
Met BC=Evapotranspiration|Gridded Source=DSS
Met BC=Evapotranspiration|Gridded Interpolation=
Met BC=Wind Speed|Expanded View=0
Met BC=Wind Speed|Point Interpolation=Nearest
Met BC=Wind Speed|Gridded Source=DSS
Met BC=Wind Speed|Gridded Interpolation=
Met BC=Wind Direction|Expanded View=0
Met BC=Wind Direction|Point Interpolation=Nearest
Met BC=Wind Direction|Gridded Source=DSS
Met BC=Wind Direction|Gridded Interpolation=
Met BC=Wind Velocity X|Expanded View=0
Met BC=Wind Velocity X|Point Interpolation=Nearest
Met BC=Wind Velocity X|Gridded Source=DSS
Met BC=Wind Velocity X|Gridded Interpolation=
Met BC=Wind Velocity Y|Expanded View=0
Met BC=Wind Velocity Y|Point Interpolation=Nearest
Met BC=Wind Velocity Y|Gridded Source=DSS
Met BC=Wind Velocity Y|Gridded Interpolation=
Met BC=Wave Forcing X|Expanded View=0
Met BC=Wave Forcing X|Point Interpolation=Nearest
Met BC=Wave Forcing X|Gridded Source=DSS
Met BC=Wave Forcing X|Gridded Interpolation=
Met BC=Wave Forcing Y|Expanded View=0
Met BC=Wave Forcing Y|Point Interpolation=Nearest
Met BC=Wave Forcing Y|Gridded Source=DSS
Met BC=Wave Forcing Y|Gridded Interpolation=
Met BC=Air Density|Mode=Constant
Met BC=Air Density|Expanded View=0
Met BC=Air Density|Constant Value=1.225
Met BC=Air Density|Constant Units=kg/m3
Met BC=Air Density|Point Interpolation=Nearest
Met BC=Air Density|Gridded Source=DSS
Met BC=Air Density|Gridded Interpolation=
Met BC=Air Temperature|Expanded View=0
Met BC=Air Temperature|Point Interpolation=Nearest
Met BC=Air Temperature|Gridded Source=DSS
Met BC=Air Temperature|Gridded Interpolation=
Met BC=Humidity|Expanded View=0
Met BC=Humidity|Point Interpolation=Nearest
Met BC=Humidity|Gridded Source=DSS
Met BC=Humidity|Gridded Interpolation=
Met BC=Air Pressure|Mode=Constant
Met BC=Air Pressure|Expanded View=0
Met BC=Air Pressure|Constant Value=1013.2
Met BC=Air Pressure|Constant Units=mb
Met BC=Air Pressure|Point Interpolation=
Met BC=Air Pressure|Gridded Source=DSS
Met BC=Air Pressure|Gridded Interpolation=
Observed Time Series=Stage|TS Name=Pipe Node: Base [15009]
Observed Time Series=Stage|TS Used=-1
Observed Time Series=Stage|TS Source=DSS
Observed Time Series=Stage|TS DSS Filename=.\SWMM Extran Datasets\EXTRAN 4 example.dss
Observed Time Series=Stage|TS DSS Pathname=/Base/15009/Stage//5Minute/EXTRAN 4 example/
Observed Time Series=Stage|TS Table Mode=0
Observed Time Series=Stage|TS Table Use Fixed Start=0
Observed Time Series=Stage|TS Table Interval=1 Hour
Observed Time Series=Stage|TS Name=Pipe Node: Base [16009]
Observed Time Series=Stage|TS Used=-1
Observed Time Series=Stage|TS Source=DSS
Observed Time Series=Stage|TS DSS Filename=.\SWMM Extran Datasets\EXTRAN 4 example.dss
Observed Time Series=Stage|TS DSS Pathname=/Base/16009/Stage//5Minute/EXTRAN 4 example/
Observed Time Series=Stage|TS Table Mode=0
Observed Time Series=Stage|TS Table Use Fixed Start=0
Observed Time Series=Stage|TS Table Interval=1 Hour
Observed Time Series=Stage|TS Name=Pipe Node: Base [16109]
Observed Time Series=Stage|TS Used=-1
Observed Time Series=Stage|TS Source=DSS
Observed Time Series=Stage|TS DSS Filename=.\SWMM Extran Datasets\EXTRAN 4 example.dss
Observed Time Series=Stage|TS DSS Pathname=/Base/16109/Stage//5Minute/EXTRAN 4 example/
Observed Time Series=Stage|TS Table Mode=0
Observed Time Series=Stage|TS Table Use Fixed Start=0
Observed Time Series=Stage|TS Table Interval=1 Hour
Observed Time Series=Stage|TS Name=Pipe Node: Base [80408]
Observed Time Series=Stage|TS Used=-1
Observed Time Series=Stage|TS Source=DSS
Observed Time Series=Stage|TS DSS Filename=.\SWMM Extran Datasets\EXTRAN 4 example.dss
Observed Time Series=Stage|TS DSS Pathname=/Base/80408/Stage//5Minute/EXTRAN 4 example/
Observed Time Series=Stage|TS Table Mode=0
Observed Time Series=Stage|TS Table Use Fixed Start=0
Observed Time Series=Stage|TS Table Interval=1 Hour
Observed Time Series=Stage|TS Name=Pipe Node: Base [80608]
Observed Time Series=Stage|TS Used=-1
Observed Time Series=Stage|TS Source=DSS
Observed Time Series=Stage|TS DSS Filename=.\SWMM Extran Datasets\EXTRAN 4 example.dss
Observed Time Series=Stage|TS DSS Pathname=/Base/80608/Stage//5Minute/EXTRAN 4 example/
Observed Time Series=Stage|TS Table Mode=0
Observed Time Series=Stage|TS Table Use Fixed Start=0
Observed Time Series=Stage|TS Table Interval=1 Hour
Observed Time Series=Stage|TS Name=Pipe Node: Base [81009]
Observed Time Series=Stage|TS Used=-1
Observed Time Series=Stage|TS Source=DSS
Observed Time Series=Stage|TS DSS Filename=.\SWMM Extran Datasets\EXTRAN 4 example.dss
Observed Time Series=Stage|TS DSS Pathname=/Base/81009/Stage//5Minute/EXTRAN 4 example/
Observed Time Series=Stage|TS Table Mode=0
Observed Time Series=Stage|TS Table Use Fixed Start=0
Observed Time Series=Stage|TS Table Interval=1 Hour
Observed Time Series=Stage|TS Name=Pipe Node: Base [81309]
Observed Time Series=Stage|TS Used=-1
Observed Time Series=Stage|TS Source=DSS
Observed Time Series=Stage|TS DSS Filename=.\SWMM Extran Datasets\EXTRAN 4 example.dss
Observed Time Series=Stage|TS DSS Pathname=/Base/81309/Stage//5Minute/EXTRAN 4 example/
Observed Time Series=Stage|TS Table Mode=0
Observed Time Series=Stage|TS Table Use Fixed Start=0
Observed Time Series=Stage|TS Table Interval=1 Hour
Observed Time Series=Stage|TS Name=Pipe Node: Base [82309]
Observed Time Series=Stage|TS Used=-1
Observed Time Series=Stage|TS Source=DSS
Observed Time Series=Stage|TS DSS Filename=.\SWMM Extran Datasets\EXTRAN 4 example.dss
Observed Time Series=Stage|TS DSS Pathname=/Base/82309/Stage//5Minute/EXTRAN 4 example/
Observed Time Series=Stage|TS Table Mode=0
Observed Time Series=Stage|TS Table Use Fixed Start=0
Observed Time Series=Stage|TS Table Interval=1 Hour
Observed Time Series=Flow|TS Name=Pipe Node: Base [15009]
Observed Time Series=Flow|TS Used=-1
Observed Time Series=Flow|TS Source=DSS
Observed Time Series=Flow|TS DSS Filename=.\SWMM Extran Datasets\EXTRAN 4 example.dss
Observed Time Series=Flow|TS DSS Pathname=/Base/15009/Flow//5Minute/EXTRAN 4 example/
Observed Time Series=Flow|TS Table Mode=0
Observed Time Series=Flow|TS Table Use Fixed Start=0
Observed Time Series=Flow|TS Table Interval=1 Hour
Observed Time Series=Flow|TS Name=Pipe Node: Base [16009]
Observed Time Series=Flow|TS Used=-1
Observed Time Series=Flow|TS Source=DSS
Observed Time Series=Flow|TS DSS Filename=.\SWMM Extran Datasets\EXTRAN 4 example.dss
Observed Time Series=Flow|TS DSS Pathname=/Base/16009/Flow//5Minute/EXTRAN 4 example/
Observed Time Series=Flow|TS Table Mode=0
Observed Time Series=Flow|TS Table Use Fixed Start=0
Observed Time Series=Flow|TS Table Interval=1 Hour
Observed Time Series=Flow|TS Name=Pipe Node: Base [16109]
Observed Time Series=Flow|TS Used=-1
Observed Time Series=Flow|TS Source=DSS
Observed Time Series=Flow|TS DSS Filename=.\SWMM Extran Datasets\EXTRAN 4 example.dss
Observed Time Series=Flow|TS DSS Pathname=/Base/16109/Flow//5Minute/EXTRAN 4 example/
Observed Time Series=Flow|TS Table Mode=0
Observed Time Series=Flow|TS Table Use Fixed Start=0
Observed Time Series=Flow|TS Table Interval=1 Hour
Observed Time Series=Flow|TS Name=Pipe Node: Base [80408]
Observed Time Series=Flow|TS Used=-1
Observed Time Series=Flow|TS Source=DSS
Observed Time Series=Flow|TS DSS Filename=.\SWMM Extran Datasets\EXTRAN 4 example.dss
Observed Time Series=Flow|TS DSS Pathname=/Base/80408/Flow//5Minute/EXTRAN 4 example/
Observed Time Series=Flow|TS Table Mode=0
Observed Time Series=Flow|TS Table Use Fixed Start=0
Observed Time Series=Flow|TS Table Interval=1 Hour
Observed Time Series=Flow|TS Name=Pipe Node: Base [80608]
Observed Time Series=Flow|TS Used=-1
Observed Time Series=Flow|TS Source=DSS
Observed Time Series=Flow|TS DSS Filename=.\SWMM Extran Datasets\EXTRAN 4 example.dss
Observed Time Series=Flow|TS DSS Pathname=/Base/80608/Flow//5Minute/EXTRAN 4 example/
Observed Time Series=Flow|TS Table Mode=0
Observed Time Series=Flow|TS Table Use Fixed Start=0
Observed Time Series=Flow|TS Table Interval=1 Hour
Observed Time Series=Flow|TS Name=Pipe Node: Base [81009]
Observed Time Series=Flow|TS Used=-1
Observed Time Series=Flow|TS Source=DSS
Observed Time Series=Flow|TS DSS Filename=.\SWMM Extran Datasets\EXTRAN 4 example.dss
Observed Time Series=Flow|TS DSS Pathname=/Base/81009/Flow//5Minute/EXTRAN 4 example/
Observed Time Series=Flow|TS Table Mode=0
Observed Time Series=Flow|TS Table Use Fixed Start=0
Observed Time Series=Flow|TS Table Interval=1 Hour
Observed Time Series=Flow|TS Name=Pipe Node: Base [81309]
Observed Time Series=Flow|TS Used=-1
Observed Time Series=Flow|TS Source=DSS
Observed Time Series=Flow|TS DSS Filename=.\SWMM Extran Datasets\EXTRAN 4 example.dss
Observed Time Series=Flow|TS DSS Pathname=/Base/81309/Flow//5Minute/EXTRAN 4 example/
Observed Time Series=Flow|TS Table Mode=0
Observed Time Series=Flow|TS Table Use Fixed Start=0
Observed Time Series=Flow|TS Table Interval=1 Hour
Observed Time Series=Flow|TS Name=Pipe Node: Base [82309]
Observed Time Series=Flow|TS Used=-1
Observed Time Series=Flow|TS Source=DSS
Observed Time Series=Flow|TS DSS Filename=.\SWMM Extran Datasets\EXTRAN 4 example.dss
Observed Time Series=Flow|TS DSS Pathname=/Base/82309/Flow//5Minute/EXTRAN 4 example/
Observed Time Series=Flow|TS Table Mode=0
Observed Time Series=Flow|TS Table Use Fixed Start=0
Observed Time Series=Flow|TS Table Interval=1 Hour
Non-Newtonian Method= 0 ,
Non-Newtonian Constant Vol Conc=0
Non-Newtonian Yield Method= 0 ,
Non-Newtonian Yield Coef=0, 0
User Yeild=   0
Non-Newtonian Sed Visc= 0 ,
Non-Newtonian Obrian B=0
User Viscosity=0
User Viscosity Ratio=0
Herschel-Bulkley Coef=0, 0
Clastic Method= 0 ,
Coulomb Phi=0
Voellmy X=0
Non-Newtonian Hindered FV= 0
Non-Newtonian FV K=0
Non-Newtonian ds=0
Non-Newtonian Max Cv=0
Non-Newtonian Bulking Method= 0 ,
Non-Newtonian High C Transport= 0 ,
Lava Activation= 0
Temperature=1300,15,,15,14,980
Heat Ballance=1,1200,0.5,1,70,0.95
Viscosity=1000,,,
Profile Coefficient=4,1.3,
Lava Param=,2500,
