HEC-RAS study ExtranTestImport.prj: SWMM Extran Tests Circular

--- ExtranTestImport.u07 (unsteady flow) ---

Flow Title=Extran 5
Program Version=7.00
Use Restart= 0
Boundary Location=                ,                ,        ,        ,                ,Perimeter 1     ,                ,DS Boundary                     ,                                ,
Friction Slope=0.0045
Boundary Location=                ,                ,        ,        ,                ,                ,                ,                                ,Base [81009]                    ,
Interval=15MIN
Flow Hydrograph= 49
       0      50      50      50      50      50      50      50      50      50
      50      50      50       0       0       0       0       0       0       0
       0       0       0       0       0       0       0       0       0       0
       0       0       0       0       0       0       0       0       0       0
       0       0       0       0       0       0       0       0       0
Stage Hydrograph TW Check=0
Use DSS=False
Use Fixed Start Time=False
Is Critical Boundary=False
Boundary Location=                ,                ,        ,        ,                ,                ,                ,                                ,Base [82309]                    ,
Interval=15MIN
Flow Hydrograph= 49
       0      40      40      40      40      40      40      40      40      40
      40      40      40       0       0       0       0       0       0       0
       0       0       0       0       0       0       0       0       0       0
       0       0       0       0       0       0       0       0       0       0
       0       0       0       0       0       0       0       0       0
Stage Hydrograph TW Check=0
Use DSS=False
Use Fixed Start Time=False
Is Critical Boundary=False
Boundary Location=                ,                ,        ,        ,                ,                ,                ,                                ,Base [80408]                    ,
Interval=15MIN
Flow Hydrograph= 49
       0      45      45      45      45      45      45      45      45      45
      45      45      45       0       0       0       0       0       0       0
       0       0       0       0       0       0       0       0       0       0
       0       0       0       0       0       0       0       0       0       0
       0       0       0       0       0       0       0       0       0
Stage Hydrograph TW Check=0
Use DSS=False
Use Fixed Start Time=False
Is Critical Boundary=False
Precipitation Mode=Disable
Wind Mode=No Wind Forces
Wave Mode=No Wave Forcing
Met BC=Precipitation|Expanded View=0
Met BC=Precipitation|Point Interpolation=Nearest
Met BC=Precipitation|Gridded Source=DSS
Met BC=Precipitation|Gridded Interpolation=
Met BC=Evapotranspiration|Expanded View=0
Met BC=Evapotranspiration|Point Interpolation=Nearest
Met BC=Evapotranspiration|Gridded Source=DSS
Met BC=Evapotranspiration|Gridded Interpolation=
Met BC=Wind Speed|Expanded View=0
Met BC=Wind Speed|Point Interpolation=Nearest
Met BC=Wind Speed|Gridded Source=DSS
Met BC=Wind Speed|Gridded Interpolation=
Met BC=Wind Direction|Expanded View=0
Met BC=Wind Direction|Point Interpolation=Nearest
Met BC=Wind Direction|Gridded Source=DSS
Met BC=Wind Direction|Gridded Interpolation=
Met BC=Wind Velocity X|Expanded View=0
Met BC=Wind Velocity X|Point Interpolation=Nearest
Met BC=Wind Velocity X|Gridded Source=DSS
Met BC=Wind Velocity X|Gridded Interpolation=
Met BC=Wind Velocity Y|Expanded View=0
Met BC=Wind Velocity Y|Point Interpolation=Nearest
Met BC=Wind Velocity Y|Gridded Source=DSS
Met BC=Wind Velocity Y|Gridded Interpolation=
Met BC=Wave Forcing X|Expanded View=0
Met BC=Wave Forcing X|Point Interpolation=Nearest
Met BC=Wave Forcing X|Gridded Source=DSS
Met BC=Wave Forcing X|Gridded Interpolation=
Met BC=Wave Forcing Y|Expanded View=0
Met BC=Wave Forcing Y|Point Interpolation=Nearest
Met BC=Wave Forcing Y|Gridded Source=DSS
Met BC=Wave Forcing Y|Gridded Interpolation=
Met BC=Air Density|Mode=Constant
Met BC=Air Density|Expanded View=0
Met BC=Air Density|Constant Value=1.225
Met BC=Air Density|Constant Units=kg/m3
Met BC=Air Density|Point Interpolation=Nearest
Met BC=Air Density|Gridded Source=DSS
Met BC=Air Density|Gridded Interpolation=
Met BC=Air Temperature|Expanded View=0
Met BC=Air Temperature|Point Interpolation=Nearest
Met BC=Air Temperature|Gridded Source=DSS
Met BC=Air Temperature|Gridded Interpolation=
Met BC=Humidity|Expanded View=0
Met BC=Humidity|Point Interpolation=Nearest
Met BC=Humidity|Gridded Source=DSS
Met BC=Humidity|Gridded Interpolation=
Met BC=Air Pressure|Mode=Constant
Met BC=Air Pressure|Expanded View=0
Met BC=Air Pressure|Constant Value=1013.2
Met BC=Air Pressure|Constant Units=mb
Met BC=Air Pressure|Point Interpolation=
Met BC=Air Pressure|Gridded Source=DSS
Met BC=Air Pressure|Gridded Interpolation=
Observed Time Series=Stage|TS Name=Pipe Node: Base [15009]
Observed Time Series=Stage|TS Used=-1
Observed Time Series=Stage|TS Source=DSS
Observed Time Series=Stage|TS DSS Filename=.\SWMM Extran Datasets\EXTRAN 5 Example.dss
Observed Time Series=Stage|TS DSS Pathname=/Base/15009/Stage//5Minute/EXTRAN 5 Example/
Observed Time Series=Stage|TS Table Mode=0
Observed Time Series=Stage|TS Table Use Fixed Start=0
Observed Time Series=Stage|TS Table StartDateTime=01Jan1988 00:00:00
Observed Time Series=Stage|TS Table Interval=1 Hour
Observed Time Series=Stage|TS Name=Pipe Node: Base [81309]
Observed Time Series=Stage|TS Used=-1
Observed Time Series=Stage|TS Source=DSS
Observed Time Series=Stage|TS DSS Filename=.\SWMM Extran Datasets\EXTRAN 5 Example.dss
Observed Time Series=Stage|TS DSS Pathname=/Base/81309/Stage//5Minute/EXTRAN 5 Example/
Observed Time Series=Stage|TS Table Mode=0
Observed Time Series=Stage|TS Table Use Fixed Start=0
Observed Time Series=Stage|TS Table StartDateTime=01Jan1988 00:00:00
Observed Time Series=Stage|TS Table Interval=1 Hour
Observed Time Series=Stage|TS Name=Pipe Node: Base [81009]
Observed Time Series=Stage|TS Used=-1
Observed Time Series=Stage|TS Source=DSS
Observed Time Series=Stage|TS DSS Filename=.\SWMM Extran Datasets\EXTRAN 5 Example.dss
Observed Time Series=Stage|TS DSS Pathname=/Base/81009/Stage//5Minute/EXTRAN 5 Example/
Observed Time Series=Stage|TS Table Mode=0
Observed Time Series=Stage|TS Table Use Fixed Start=0
Observed Time Series=Stage|TS Table StartDateTime=01Jan1988 00:00:00
Observed Time Series=Stage|TS Table Interval=1 Hour
Observed Time Series=Stage|TS Name=Pipe Node: Base [16109]
Observed Time Series=Stage|TS Used=-1
Observed Time Series=Stage|TS Source=DSS
Observed Time Series=Stage|TS DSS Filename=.\SWMM Extran Datasets\EXTRAN 5 Example.dss
Observed Time Series=Stage|TS DSS Pathname=/Base/16109/Stage//5Minute/EXTRAN 5 Example/
Observed Time Series=Stage|TS Table Mode=0
Observed Time Series=Stage|TS Table Use Fixed Start=0
Observed Time Series=Stage|TS Table StartDateTime=01Jan1988 00:00:00
Observed Time Series=Stage|TS Table Interval=1 Hour
Observed Time Series=Stage|TS Name=Pipe Node: Base [82309]
Observed Time Series=Stage|TS Used=-1
Observed Time Series=Stage|TS Source=DSS
Observed Time Series=Stage|TS DSS Filename=.\SWMM Extran Datasets\EXTRAN 5 Example.dss
Observed Time Series=Stage|TS DSS Pathname=/Base/82309/Stage//5Minute/EXTRAN 5 Example/
Observed Time Series=Stage|TS Table Mode=0
Observed Time Series=Stage|TS Table Use Fixed Start=0
Observed Time Series=Stage|TS Table StartDateTime=01Jan1988 00:00:00
Observed Time Series=Stage|TS Table Interval=1 Hour
Observed Time Series=Stage|TS Name=Pipe Node: Base [80608]
Observed Time Series=Stage|TS Used=-1
Observed Time Series=Stage|TS Source=DSS
Observed Time Series=Stage|TS DSS Filename=.\SWMM Extran Datasets\EXTRAN 5 Example.dss
Observed Time Series=Stage|TS DSS Pathname=/Base/80608/Stage//5Minute/EXTRAN 5 Example/
Observed Time Series=Stage|TS Table Mode=0
Observed Time Series=Stage|TS Table Use Fixed Start=0
Observed Time Series=Stage|TS Table StartDateTime=01Jan1988 00:00:00
Observed Time Series=Stage|TS Table Interval=1 Hour
Observed Time Series=Stage|TS Name=Pipe Node: Base [80408]
Observed Time Series=Stage|TS Used=-1
Observed Time Series=Stage|TS Source=DSS
Observed Time Series=Stage|TS DSS Filename=.\SWMM Extran Datasets\EXTRAN 5 Example.dss
Observed Time Series=Stage|TS DSS Pathname=/Base/80408/Stage//5Minute/EXTRAN 5 Example/
Observed Time Series=Stage|TS Table Mode=0
Observed Time Series=Stage|TS Table Use Fixed Start=0
Observed Time Series=Stage|TS Table Interval=1 Hour
Observed Time Series=Stage|TS Name=Pipe Node: Base [16009]
Observed Time Series=Stage|TS Used=-1
Observed Time Series=Stage|TS Source=DSS
Observed Time Series=Stage|TS DSS Filename=.\SWMM Extran Datasets\EXTRAN 5 Example.dss
Observed Time Series=Stage|TS DSS Pathname=/Base/16009/Stage//5Minute/EXTRAN 5 Example/
Observed Time Series=Stage|TS Table Mode=0
Observed Time Series=Stage|TS Table Use Fixed Start=0
Observed Time Series=Stage|TS Table Interval=1 Hour
Observed Time Series=Stage|TS Name=Pipe Node: Base [82308]
Observed Time Series=Stage|TS Used=-1
Observed Time Series=Stage|TS Source=DSS
Observed Time Series=Stage|TS DSS Filename=.\SWMM Extran Datasets\EXTRAN 5 Example.dss
Observed Time Series=Stage|TS DSS Pathname=/Base/82308/Stage//5Minute/EXTRAN 5 Example/
Observed Time Series=Stage|TS Table Mode=0
Observed Time Series=Stage|TS Table Use Fixed Start=0
Observed Time Series=Stage|TS Table Interval=1 Hour
Observed Time Series=Flow|TS Name=Pipe Node: Base [15009]
Observed Time Series=Flow|TS Used=-1
Observed Time Series=Flow|TS Source=DSS
Observed Time Series=Flow|TS DSS Filename=.\SWMM Extran Datasets\EXTRAN 5 Example.dss
Observed Time Series=Flow|TS DSS Pathname=/Base/15009/Flow//5Minute/EXTRAN 5 Example/
Observed Time Series=Flow|TS Table Mode=0
Observed Time Series=Flow|TS Table Use Fixed Start=0
Observed Time Series=Flow|TS Table Interval=1 Hour
Observed Time Series=Flow|TS Name=Pipe Node: Base [16009]
Observed Time Series=Flow|TS Used=-1
Observed Time Series=Flow|TS Source=DSS
Observed Time Series=Flow|TS DSS Filename=.\SWMM Extran Datasets\EXTRAN 5 Example.dss
Observed Time Series=Flow|TS DSS Pathname=/Base/16009/Flow//5Minute/EXTRAN 5 Example/
Observed Time Series=Flow|TS Table Mode=0
Observed Time Series=Flow|TS Table Use Fixed Start=0
Observed Time Series=Flow|TS Table Interval=1 Hour
Observed Time Series=Flow|TS Name=Pipe Node: Base [16109]
Observed Time Series=Flow|TS Used=-1
Observed Time Series=Flow|TS Source=DSS
Observed Time Series=Flow|TS DSS Filename=.\SWMM Extran Datasets\EXTRAN 5 Example.dss
Observed Time Series=Flow|TS DSS Pathname=/Base/16109/Flow//5Minute/EXTRAN 5 Example/
Observed Time Series=Flow|TS Table Mode=0
Observed Time Series=Flow|TS Table Use Fixed Start=0
Observed Time Series=Flow|TS Table Interval=1 Hour
Observed Time Series=Flow|TS Name=Pipe Node: Base [80408]
Observed Time Series=Flow|TS Used=-1
Observed Time Series=Flow|TS Source=DSS
Observed Time Series=Flow|TS DSS Filename=.\SWMM Extran Datasets\EXTRAN 5 Example.dss
Observed Time Series=Flow|TS DSS Pathname=/Base/80408/Flow//5Minute/EXTRAN 5 Example/
Observed Time Series=Flow|TS Table Mode=0
Observed Time Series=Flow|TS Table Use Fixed Start=0
Observed Time Series=Flow|TS Table Interval=1 Hour
Observed Time Series=Flow|TS Name=Pipe Node: Base [80608]
Observed Time Series=Flow|TS Used=-1
Observed Time Series=Flow|TS Source=DSS
Observed Time Series=Flow|TS DSS Filename=.\SWMM Extran Datasets\EXTRAN 5 Example.dss
Observed Time Series=Flow|TS DSS Pathname=/Base/80608/Flow//5Minute/EXTRAN 5 Example/
Observed Time Series=Flow|TS Table Mode=0
Observed Time Series=Flow|TS Table Use Fixed Start=0
Observed Time Series=Flow|TS Table Interval=1 Hour
Observed Time Series=Flow|TS Name=Pipe Node: Base [81009]
Observed Time Series=Flow|TS Used=-1
Observed Time Series=Flow|TS Source=DSS
Observed Time Series=Flow|TS DSS Filename=.\SWMM Extran Datasets\EXTRAN 5 Example.dss
Observed Time Series=Flow|TS DSS Pathname=/Base/81009/Flow//5Minute/EXTRAN 5 Example/
Observed Time Series=Flow|TS Table Mode=0
Observed Time Series=Flow|TS Table Use Fixed Start=0
Observed Time Series=Flow|TS Table Interval=1 Hour
Observed Time Series=Flow|TS Name=Pipe Node: Base [81309]
Observed Time Series=Flow|TS Used=-1
Observed Time Series=Flow|TS Source=DSS
Observed Time Series=Flow|TS DSS Filename=.\SWMM Extran Datasets\EXTRAN 5 Example.dss
Observed Time Series=Flow|TS DSS Pathname=/Base/81309/Flow//5Minute/EXTRAN 5 Example/
Observed Time Series=Flow|TS Table Mode=0
Observed Time Series=Flow|TS Table Use Fixed Start=0
Observed Time Series=Flow|TS Table Interval=1 Hour
Observed Time Series=Flow|TS Name=Pipe Node: Base [82309]
Observed Time Series=Flow|TS Used=-1
Observed Time Series=Flow|TS Source=DSS
Observed Time Series=Flow|TS DSS Filename=.\SWMM Extran Datasets\EXTRAN 5 Example.dss
Observed Time Series=Flow|TS DSS Pathname=/Base/82309/Flow//5Minute/EXTRAN 5 Example/
Observed Time Series=Flow|TS Table Mode=0
Observed Time Series=Flow|TS Table Use Fixed Start=0
Observed Time Series=Flow|TS Table Interval=1 Hour
Observed Time Series=Flow|TS Name=Pipe Node: Base [82308]
Observed Time Series=Flow|TS Used=-1
Observed Time Series=Flow|TS Source=DSS
Observed Time Series=Flow|TS DSS Filename=.\SWMM Extran Datasets\EXTRAN 5 Example.dss
Observed Time Series=Flow|TS DSS Pathname=/Base/82308/Flow//5Minute/EXTRAN 5 Example/
Observed Time Series=Flow|TS Table Mode=0
Observed Time Series=Flow|TS Table Use Fixed Start=0
Observed Time Series=Flow|TS Table Interval=1 Hour
Non-Newtonian Method= 0 ,
Non-Newtonian Constant Vol Conc=0
Non-Newtonian Yield Method= 0 ,
Non-Newtonian Yield Coef=0, 0
User Yeild=   0
Non-Newtonian Sed Visc= 0 ,
Non-Newtonian Obrian B=0
User Viscosity=0
User Viscosity Ratio=0
Herschel-Bulkley Coef=0, 0
Clastic Method= 0 ,
Coulomb Phi=0
Voellmy X=0
Non-Newtonian Hindered FV= 0
Non-Newtonian FV K=0
Non-Newtonian ds=0
Non-Newtonian Max Cv=0
Non-Newtonian Bulking Method= 0 ,
Non-Newtonian High C Transport= 0 ,
Lava Activation= 0
Temperature=1300,15,,15,14,980
Heat Ballance=1,1200,0.5,1,70,0.95
Viscosity=1000,,,
Profile Coefficient=4,1.3,
Lava Param=,2500,

--- ExtranTestImport.u08 (unsteady flow) ---

Flow Title=Extran 4 Rating Cruive
Program Version=7.00
Use Restart= 0
Boundary Location=                ,                ,        ,        ,                ,Perimeter 1     ,                ,DS Boundary                     ,                                ,
Friction Slope=0.0045
Boundary Location=                ,                ,        ,        ,                ,                ,                ,                                ,Base [81009]                    ,
Interval=15MIN
Flow Hydrograph= 49
       0       2       4       6       8      10      12      14      16      18
      20      22      24      26      28      30      32      34      36      38
      40      42      44      46      48      50      52      54      56      58
      60      62      64      66      68      70      72      74      76      78
      80      82      84      86      88      90       0       0       0
Stage Hydrograph TW Check=0
Use DSS=False
Use Fixed Start Time=False
Is Critical Boundary=False
Boundary Location=                ,                ,        ,        ,                ,                ,                ,                                ,Base [82309]                    ,
Interval=15MIN
Flow Hydrograph= 49
       0   2.105   4.211   6.316   8.421  10.526  12.632  14.737  16.842  18.947
  21.053  23.158  25.263  27.368  29.474  31.579  33.684  35.789  37.895      40
  38.462  36.923  35.385  33.846  32.308  30.769  29.231  27.692  26.154  24.615
  23.077  21.538      20  18.462  16.923  15.385  13.846  12.308  10.769   9.231
   7.692   6.154   4.615   3.077   1.538       0       0       0       0
Stage Hydrograph TW Check=0
Use DSS=False
Use Fixed Start Time=False
Is Critical Boundary=False
Boundary Location=                ,                ,        ,        ,                ,                ,                ,                                ,Base [80408]                    ,
Interval=15MIN
Flow Hydrograph= 49
       0      45      45      45      45      45      45      45      45      45
      45      45      45       0       0       0       0       0       0       0
       0       0       0       0       0       0       0       0       0       0
       0       0       0       0       0       0       0       0       0       0
       0       0       0       0       0       0       0       0       0
Stage Hydrograph TW Check=0
Use DSS=False
Use Fixed Start Time=False
Is Critical Boundary=False
Precipitation Mode=Disable
Wind Mode=No Wind Forces
Wave Mode=No Wave Forcing
Met BC=Precipitation|Expanded View=0
Met BC=Precipitation|Point Interpolation=Nearest
Met BC=Precipitation|Gridded Source=DSS
Met BC=Precipitation|Gridded Interpolation=
Met BC=Evapotranspiration|Expanded View=0
Met BC=Evapotranspiration|Point Interpolation=Nearest
Met BC=Evapotranspiration|Gridded Source=DSS
Met BC=Evapotranspiration|Gridded Interpolation=
Met BC=Wind Speed|Expanded View=0
Met BC=Wind Speed|Point Interpolation=Nearest
Met BC=Wind Speed|Gridded Source=DSS
Met BC=Wind Speed|Gridded Interpolation=
Met BC=Wind Direction|Expanded View=0
Met BC=Wind Direction|Point Interpolation=Nearest
Met BC=Wind Direction|Gridded Source=DSS
Met BC=Wind Direction|Gridded Interpolation=
Met BC=Wind Velocity X|Expanded View=0
Met BC=Wind Velocity X|Point Interpolation=Nearest
Met BC=Wind Velocity X|Gridded Source=DSS
Met BC=Wind Velocity X|Gridded Interpolation=
Met BC=Wind Velocity Y|Expanded View=0
Met BC=Wind Velocity Y|Point Interpolation=Nearest
Met BC=Wind Velocity Y|Gridded Source=DSS
Met BC=Wind Velocity Y|Gridded Interpolation=
Met BC=Wave Forcing X|Expanded View=0
Met BC=Wave Forcing X|Point Interpolation=Nearest
Met BC=Wave Forcing X|Gridded Source=DSS
Met BC=Wave Forcing X|Gridded Interpolation=
Met BC=Wave Forcing Y|Expanded View=0
Met BC=Wave Forcing Y|Point Interpolation=Nearest
Met BC=Wave Forcing Y|Gridded Source=DSS
Met BC=Wave Forcing Y|Gridded Interpolation=
Met BC=Air Density|Mode=Constant
Met BC=Air Density|Expanded View=0
Met BC=Air Density|Constant Value=1.225
Met BC=Air Density|Constant Units=kg/m3
Met BC=Air Density|Point Interpolation=Nearest
Met BC=Air Density|Gridded Source=DSS
Met BC=Air Density|Gridded Interpolation=
Met BC=Air Temperature|Expanded View=0
Met BC=Air Temperature|Point Interpolation=Nearest
Met BC=Air Temperature|Gridded Source=DSS
Met BC=Air Temperature|Gridded Interpolation=
Met BC=Humidity|Expanded View=0
Met BC=Humidity|Point Interpolation=Nearest
Met BC=Humidity|Gridded Source=DSS
Met BC=Humidity|Gridded Interpolation=
Met BC=Air Pressure|Mode=Constant
Met BC=Air Pressure|Expanded View=0
Met BC=Air Pressure|Constant Value=1013.2
Met BC=Air Pressure|Constant Units=mb
Met BC=Air Pressure|Point Interpolation=
Met BC=Air Pressure|Gridded Source=DSS
Met BC=Air Pressure|Gridded Interpolation=
Observed Time Series=Stage|TS Name=Pipe Node: Base [15009]
Observed Time Series=Stage|TS Used=-1
Observed Time Series=Stage|TS Source=DSS
Observed Time Series=Stage|TS DSS Filename=.\SWMM Extran Datasets\EXTRAN 5 Example.dss
Observed Time Series=Stage|TS DSS Pathname=/Base/15009/Stage//5Minute/EXTRAN 5 Example/
Observed Time Series=Stage|TS Table Mode=0
Observed Time Series=Stage|TS Table Use Fixed Start=0
Observed Time Series=Stage|TS Table Interval=1 Hour
Observed Time Series=Stage|TS Name=Pipe Node: Base [16009]
Observed Time Series=Stage|TS Used=-1
Observed Time Series=Stage|TS Source=DSS
Observed Time Series=Stage|TS DSS Filename=.\SWMM Extran Datasets\EXTRAN 5 Example.dss
Observed Time Series=Stage|TS DSS Pathname=/Base/16009/Stage//5Minute/EXTRAN 5 Example/
Observed Time Series=Stage|TS Table Mode=0
Observed Time Series=Stage|TS Table Use Fixed Start=0
Observed Time Series=Stage|TS Table Interval=1 Hour
Observed Time Series=Stage|TS Name=Pipe Node: Base [16109]
Observed Time Series=Stage|TS Used=-1
Observed Time Series=Stage|TS Source=DSS
Observed Time Series=Stage|TS DSS Filename=.\SWMM Extran Datasets\EXTRAN 5 Example.dss
Observed Time Series=Stage|TS DSS Pathname=/Base/16109/Stage//5Minute/EXTRAN 5 Example/
Observed Time Series=Stage|TS Table Mode=0
Observed Time Series=Stage|TS Table Use Fixed Start=0
Observed Time Series=Stage|TS Table Interval=1 Hour
Observed Time Series=Stage|TS Name=Pipe Node: Base [80408]
Observed Time Series=Stage|TS Used=-1
Observed Time Series=Stage|TS Source=DSS
Observed Time Series=Stage|TS DSS Filename=.\SWMM Extran Datasets\EXTRAN 5 Example.dss
Observed Time Series=Stage|TS DSS Pathname=/Base/80408/Stage//5Minute/EXTRAN 5 Example/
Observed Time Series=Stage|TS Table Mode=0
Observed Time Series=Stage|TS Table Use Fixed Start=0
Observed Time Series=Stage|TS Table Interval=1 Hour
Observed Time Series=Stage|TS Name=Pipe Node: Base [80608]
Observed Time Series=Stage|TS Used=-1
Observed Time Series=Stage|TS Source=DSS
Observed Time Series=Stage|TS DSS Filename=.\SWMM Extran Datasets\EXTRAN 5 Example.dss
Observed Time Series=Stage|TS DSS Pathname=/Base/80608/Stage//5Minute/EXTRAN 5 Example/
Observed Time Series=Stage|TS Table Mode=0
Observed Time Series=Stage|TS Table Use Fixed Start=0
Observed Time Series=Stage|TS Table Interval=1 Hour
Observed Time Series=Stage|TS Name=Pipe Node: Base [81009]
Observed Time Series=Stage|TS Used=-1
Observed Time Series=Stage|TS Source=DSS
Observed Time Series=Stage|TS DSS Filename=.\SWMM Extran Datasets\EXTRAN 5 Example.dss
Observed Time Series=Stage|TS DSS Pathname=/Base/81009/Stage//5Minute/EXTRAN 5 Example/
Observed Time Series=Stage|TS Table Mode=0
Observed Time Series=Stage|TS Table Use Fixed Start=0
Observed Time Series=Stage|TS Table Interval=1 Hour
Observed Time Series=Stage|TS Name=Pipe Node: Base [81309]
Observed Time Series=Stage|TS Used=-1
Observed Time Series=Stage|TS Source=DSS
Observed Time Series=Stage|TS DSS Filename=.\SWMM Extran Datasets\EXTRAN 5 Example.dss
Observed Time Series=Stage|TS DSS Pathname=/Base/81309/Stage//5Minute/EXTRAN 5 Example/
Observed Time Series=Stage|TS Table Mode=0
Observed Time Series=Stage|TS Table Use Fixed Start=0
Observed Time Series=Stage|TS Table Interval=1 Hour
Observed Time Series=Stage|TS Name=Pipe Node: Base [82309]
Observed Time Series=Stage|TS Used=-1
Observed Time Series=Stage|TS Source=DSS
Observed Time Series=Stage|TS DSS Filename=.\SWMM Extran Datasets\EXTRAN 5 Example.dss
Observed Time Series=Stage|TS DSS Pathname=/Base/82309/Stage//5Minute/EXTRAN 5 Example/
Observed Time Series=Stage|TS Table Mode=0
Observed Time Series=Stage|TS Table Use Fixed Start=0
Observed Time Series=Stage|TS Table Interval=1 Hour
Observed Time Series=Flow|TS Name=Pipe Node: Base [15009]
Observed Time Series=Flow|TS Used=-1
Observed Time Series=Flow|TS Source=DSS
Observed Time Series=Flow|TS DSS Filename=.\SWMM Extran Datasets\EXTRAN 5 Example.dss
Observed Time Series=Flow|TS DSS Pathname=/Base/15009/Flow//5Minute/EXTRAN 5 Example/
Observed Time Series=Flow|TS Table Mode=0
Observed Time Series=Flow|TS Table Use Fixed Start=0
Observed Time Series=Flow|TS Table Interval=1 Hour
Observed Time Series=Flow|TS Name=Pipe Node: Base [16009]
Observed Time Series=Flow|TS Used=-1
Observed Time Series=Flow|TS Source=DSS
Observed Time Series=Flow|TS DSS Filename=.\SWMM Extran Datasets\EXTRAN 5 Example.dss
Observed Time Series=Flow|TS DSS Pathname=/Base/16009/Flow//5Minute/EXTRAN 5 Example/
Observed Time Series=Flow|TS Table Mode=0
Observed Time Series=Flow|TS Table Use Fixed Start=0
Observed Time Series=Flow|TS Table Interval=1 Hour
Observed Time Series=Flow|TS Name=Pipe Node: Base [16109]
Observed Time Series=Flow|TS Used=-1
Observed Time Series=Flow|TS Source=DSS
Observed Time Series=Flow|TS DSS Filename=.\SWMM Extran Datasets\EXTRAN 5 Example.dss
Observed Time Series=Flow|TS DSS Pathname=/Base/16109/Flow//5Minute/EXTRAN 5 Example/
Observed Time Series=Flow|TS Table Mode=0
Observed Time Series=Flow|TS Table Use Fixed Start=0
Observed Time Series=Flow|TS Table Interval=1 Hour
Observed Time Series=Flow|TS Name=Pipe Node: Base [80408]
Observed Time Series=Flow|TS Used=-1
Observed Time Series=Flow|TS Source=DSS
Observed Time Series=Flow|TS DSS Filename=.\SWMM Extran Datasets\EXTRAN 5 Example.dss
Observed Time Series=Flow|TS DSS Pathname=/Base/80408/Flow//5Minute/EXTRAN 5 Example/
Observed Time Series=Flow|TS Table Mode=0
Observed Time Series=Flow|TS Table Use Fixed Start=0
Observed Time Series=Flow|TS Table Interval=1 Hour
Observed Time Series=Flow|TS Name=Pipe Node: Base [80608]
Observed Time Series=Flow|TS Used=-1
Observed Time Series=Flow|TS Source=DSS
Observed Time Series=Flow|TS DSS Filename=.\SWMM Extran Datasets\EXTRAN 5 Example.dss
Observed Time Series=Flow|TS DSS Pathname=/Base/80608/Flow//5Minute/EXTRAN 5 Example/
Observed Time Series=Flow|TS Table Mode=0
Observed Time Series=Flow|TS Table Use Fixed Start=0
Observed Time Series=Flow|TS Table Interval=1 Hour
Observed Time Series=Flow|TS Name=Pipe Node: Base [81009]
Observed Time Series=Flow|TS Used=-1
Observed Time Series=Flow|TS Source=DSS
Observed Time Series=Flow|TS DSS Filename=.\SWMM Extran Datasets\EXTRAN 5 Example.dss
Observed Time Series=Flow|TS DSS Pathname=/Base/81009/Flow//5Minute/EXTRAN 5 Example/
Observed Time Series=Flow|TS Table Mode=0
Observed Time Series=Flow|TS Table Use Fixed Start=0
Observed Time Series=Flow|TS Table Interval=1 Hour
Observed Time Series=Flow|TS Name=Pipe Node: Base [81309]
Observed Time Series=Flow|TS Used=-1
Observed Time Series=Flow|TS Source=DSS
Observed Time Series=Flow|TS DSS Filename=.\SWMM Extran Datasets\EXTRAN 5 Example.dss
Observed Time Series=Flow|TS DSS Pathname=/Base/81309/Flow//5Minute/EXTRAN 5 Example/
Observed Time Series=Flow|TS Table Mode=0
Observed Time Series=Flow|TS Table Use Fixed Start=0
Observed Time Series=Flow|TS Table Interval=1 Hour
Observed Time Series=Flow|TS Name=Pipe Node: Base [82309]
Observed Time Series=Flow|TS Used=-1
Observed Time Series=Flow|TS Source=DSS
Observed Time Series=Flow|TS DSS Filename=.\SWMM Extran Datasets\EXTRAN 5 Example.dss
Observed Time Series=Flow|TS DSS Pathname=/Base/82309/Flow//5Minute/EXTRAN 5 Example/
Observed Time Series=Flow|TS Table Mode=0
Observed Time Series=Flow|TS Table Use Fixed Start=0
Observed Time Series=Flow|TS Table Interval=1 Hour
Non-Newtonian Method= 0 ,
Non-Newtonian Constant Vol Conc=0
Non-Newtonian Yield Method= 0 ,
Non-Newtonian Yield Coef=0, 0
User Yeild=   0
Non-Newtonian Sed Visc= 0 ,
Non-Newtonian Obrian B=0
User Viscosity=0
User Viscosity Ratio=0
Herschel-Bulkley Coef=0, 0
Clastic Method= 0 ,
Coulomb Phi=0
Voellmy X=0
Non-Newtonian Hindered FV= 0
Non-Newtonian FV K=0
Non-Newtonian ds=0
Non-Newtonian Max Cv=0
Non-Newtonian Bulking Method= 0 ,
Non-Newtonian High C Transport= 0 ,
Lava Activation= 0
Temperature=1300,15,,15,14,980
Heat Ballance=1,1200,0.5,1,70,0.95
Viscosity=1000,,,
Profile Coefficient=4,1.3,
Lava Param=,2500,

--- ExtranTestImport.g07 (geometry) ---

Geom Title=Extran 7 - InlinePump
Program Version=7.00

Storage Area=Perimeter 1     ,10443.3929315,4277.3286068
Storage Area Surface Line= 6
11708.27876512332388.92591623079
11023.89661551352444.81959492957
9522.339776481886640.06528495057
9578.792581457296659.99005339071
11078.73399742812469.65776642782
11708.27876512332388.92591623079
Storage Area Type= 1
Storage Area Is2D=-1
Storage Area Point Generation Data=,,50,50
Storage Area 2D Points= 31
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Storage Area Mannings=0.015
2D Cell Volume Filter Tolerance=0.01
2D Cell Minimum Area Fraction=0.01
2D Face Profile Filter Tolerance=0.01
2D Face Area Elevation Profile Filter Tolerance=0.01
2D Face Area Elevation Conveyance Ratio=0.02
2D Face Min Length Ratio=0.05
2D Face Area Laminar Depth=0.2
2D Multiple Face Mann n=0
2D Composite LC=0

BC Line Name=DS Boundary
BC Line Storage Area=Perimeter 1
BC Line Start Position= 9522.59932215836 , 6644.19892020173
BC Line Middle Position= 9548.47627047713 , 6653.14803149531
BC Line End Position= 9574.35321879591 , 6662.09714278889
BC Line Arc= 2
9522.599322158366644.198920201739574.353218795916662.09714278889

Pump Station=Pump Station #1 ,16694.3759398,2679.9117202,,,16694.3759398,2679.9117202
Pump Station From=                ,                ,        ,                ,,Base [82309]
Pump Station To=                ,                ,        ,                ,,Base [15009]
Pump Station TW Min=112.3
Pump Station Group=Group #1        ,False,5,5,4
Pump Station Group Pump=Pump #1         ,115,112.7
Pump Station Group Pump Centerline= 2
16689.46479540322921.0339773014916689.47433659162421.05567836401
Pump Station Group HQ= 2
       0       0     100     100
LCMann Table=0

Chan Stop Cuts=-1
Use User Specified Reach Order=0
Composite Channel Slope=5

--- ExtranTestImport.g01 (geometry) ---

Geom Title=Extran 4 - Weir
Program Version=7.00

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
Storage Area=Perimeter 1     ,,
Storage Area Surface Line= 6
11708.27876512332388.92591623079
11023.89661551352444.81959492957
9522.339776481886640.06528495057
9578.792581457296659.99005339071
11078.73399742812469.65776642782
11708.27876512332388.92591623079
Storage Area Type= 1
Storage Area Is2D=-1
Storage Area Point Generation Data=,,154.2524,154.2524
Storage Area 2D Points= 32
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Storage Area Mannings=0.015
2D Cell Volume Filter Tolerance=0.01
2D Cell Minimum Area Fraction=0.01
2D Face Profile Filter Tolerance=0.01
2D Face Area Elevation Profile Filter Tolerance=0.01
2D Face Area Elevation Conveyance Ratio=0.02
2D Face Min Length Ratio=0.05
2D Face Area Laminar Depth=0.2
2D Multiple Face Mann n=0
2D Composite LC=0

Storage Area=Surface Stor 1  ,,
Storage Area Surface Line= 6
20562.46993231352973.35268498287
20504.88853190692973.28935054041
 20503.9658789023164.15629239523
20566.5408499143 3164.3132664507
20566.43626682572918.94633386912
20562.46993231352973.35268498287
Storage Area Type= 1
Storage Area Is2D=-1
Storage Area Point Generation Data=0,0,46.45469,46.45469
Storage Area 2D Points= 2
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Storage Area Mannings=0.06
2D Cell Volume Filter Tolerance=0.01
2D Cell Minimum Area Fraction=0.01
2D Face Profile Filter Tolerance=0.01
2D Face Area Elevation Profile Filter Tolerance=0.01
2D Face Area Elevation Conveyance Ratio=0.02
2D Face Min Length Ratio=0.05
2D Face Area Laminar Depth=0.2
2D Multiple Face Mann n=0
2D Composite LC=0

Storage Area=Surface Stor 2  ,,
Storage Area Surface Line= 6
18762.98642899792973.31467001867
18705.40502859132973.25133557621
18706.09970723033165.73560907496
18768.67467824263165.89258313043
18766.95276351012918.90831890492
18762.98642899792973.31467001867
Storage Area Type= 1
Storage Area Is2D=-1
Storage Area Point Generation Data=0,0,42.86091,42.86091
Storage Area 2D Points= 2
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Storage Area Mannings=0.06
2D Cell Volume Filter Tolerance=0.01
2D Cell Minimum Area Fraction=0.01
2D Face Profile Filter Tolerance=0.01
2D Face Area Elevation Profile Filter Tolerance=0.01
2D Face Area Elevation Conveyance Ratio=0.02
2D Face Min Length Ratio=0.05
2D Face Area Laminar Depth=0.2
2D Multiple Face Mann n=0
2D Composite LC=0

BC Line Name=DS Boundary
BC Line Storage Area=Perimeter 1
BC Line Start Position= 9522.59932215836 , 6644.19892020173
BC Line Middle Position= 9548.47627047713 , 6653.14803149531
BC Line End Position= 9574.35321879591 , 6662.09714278889
BC Line Arc= 2
9522.599322158366644.198920201739574.353218795916662.09714278889
LCMann Table=0

--- ExtranTestImport.g02 (geometry) ---

Geom Title=Extran 1 and 2
Program Version=7.00

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
Storage Area=Perimeter 1     ,,
Storage Area Surface Line= 6
11708.27876512332388.92591623079
11023.89661551352444.81959492957
9522.339776481886640.06528495057
9578.792581457296659.99005339071
11078.73399742812469.65776642782
11708.27876512332388.92591623079
Storage Area Type= 1
Storage Area Is2D=-1
Storage Area Point Generation Data=,,154.2524,154.2524
Storage Area 2D Points= 32
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Storage Area Mannings=0.015
2D Cell Volume Filter Tolerance=0.01
2D Cell Minimum Area Fraction=0.01
2D Face Profile Filter Tolerance=0.01
2D Face Area Elevation Profile Filter Tolerance=0.01
2D Face Area Elevation Conveyance Ratio=0.02
2D Face Min Length Ratio=0.05
2D Face Area Laminar Depth=0.2
2D Multiple Face Mann n=0
2D Composite LC=0

Storage Area=Surface Stor 1  ,,
Storage Area Surface Line= 6
20562.46993231352973.35268498287
20504.88853190692973.28935054041
 20503.9658789023164.15629239523
20566.5408499143 3164.3132664507
20566.43626682572918.94633386912
20562.46993231352973.35268498287
Storage Area Type= 1
Storage Area Is2D=-1
Storage Area Point Generation Data=0,0,46.45469,46.45469
Storage Area 2D Points= 2
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Storage Area Mannings=0.06
2D Cell Volume Filter Tolerance=0.01
2D Cell Minimum Area Fraction=0.01
2D Face Profile Filter Tolerance=0.01
2D Face Area Elevation Profile Filter Tolerance=0.01
2D Face Area Elevation Conveyance Ratio=0.02
2D Face Min Length Ratio=0.05
2D Face Area Laminar Depth=0.2
2D Multiple Face Mann n=0
2D Composite LC=0

Storage Area=Surface Stor 2  ,,
Storage Area Surface Line= 6
18762.98642899792973.31467001867
18705.40502859132973.25133557621
18706.09970723033165.73560907496
18768.67467824263165.89258313043
18766.95276351012918.90831890492
18762.98642899792973.31467001867
Storage Area Type= 1
Storage Area Is2D=-1
Storage Area Point Generation Data=0,0,42.86091,42.86091
Storage Area 2D Points= 2
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Storage Area Mannings=0.06
2D Cell Volume Filter Tolerance=0.01
2D Cell Minimum Area Fraction=0.01
2D Face Profile Filter Tolerance=0.01
2D Face Area Elevation Profile Filter Tolerance=0.01
2D Face Area Elevation Conveyance Ratio=0.02
2D Face Min Length Ratio=0.05
2D Face Area Laminar Depth=0.2
2D Multiple Face Mann n=0
2D Composite LC=0

BC Line Name=DS Boundary
BC Line Storage Area=Perimeter 1
BC Line Start Position= 9522.59932215836 , 6644.19892020173
BC Line Middle Position= 9548.47627047713 , 6653.14803149531
BC Line End Position= 9574.35321879591 , 6662.09714278889
BC Line Arc= 2
9522.599322158366644.198920201739574.353218795916662.09714278889
LCMann Table=0

--- ExtranTestImport.g04 (geometry) ---

Geom Title=Extran 5 -Side  Orifice
Program Version=7.00

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
Storage Area=Perimeter 1     ,,
Storage Area Surface Line= 6
11708.27876512332388.92591623079
11023.89661551352444.81959492957
9522.339776481886640.06528495057
9578.792581457296659.99005339071
11078.73399742812469.65776642782
11708.27876512332388.92591623079
Storage Area Type= 1
Storage Area Is2D=-1
Storage Area Point Generation Data=,,154.2524,154.2524
Storage Area 2D Points= 32
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Storage Area Mannings=0.015
2D Cell Volume Filter Tolerance=0.01
2D Cell Minimum Area Fraction=0.01
2D Face Profile Filter Tolerance=0.01
2D Face Area Elevation Profile Filter Tolerance=0.01
2D Face Area Elevation Conveyance Ratio=0.02
2D Face Min Length Ratio=0.05
2D Face Area Laminar Depth=0.2
2D Multiple Face Mann n=0
2D Composite LC=0

Storage Area=Surface Stor 1  ,,
Storage Area Surface Line= 6
20562.46993231352973.35268498287
20504.88853190692973.28935054041
 20503.9658789023164.15629239523
20566.5408499143 3164.3132664507
20566.43626682572918.94633386912
20562.46993231352973.35268498287
Storage Area Type= 1
Storage Area Is2D=-1
Storage Area Point Generation Data=0,0,46.45469,46.45469
Storage Area 2D Points= 2
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Storage Area Mannings=0.06
2D Cell Volume Filter Tolerance=0.01
2D Cell Minimum Area Fraction=0.01
2D Face Profile Filter Tolerance=0.01
2D Face Area Elevation Profile Filter Tolerance=0.01
2D Face Area Elevation Conveyance Ratio=0.02
2D Face Min Length Ratio=0.05
2D Face Area Laminar Depth=0.2
2D Multiple Face Mann n=0
2D Composite LC=0

Storage Area=Surface Stor 2  ,,
Storage Area Surface Line= 6
18762.98642899792973.31467001867
18705.40502859132973.25133557621
18706.09970723033165.73560907496
18768.67467824263165.89258313043
18766.95276351012918.90831890492
18762.98642899792973.31467001867
Storage Area Type= 1
Storage Area Is2D=-1
Storage Area Point Generation Data=0,0,42.86091,42.86091
Storage Area 2D Points= 2
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Storage Area Mannings=0.06
2D Cell Volume Filter Tolerance=0.01
2D Cell Minimum Area Fraction=0.01
2D Face Profile Filter Tolerance=0.01
2D Face Area Elevation Profile Filter Tolerance=0.01
2D Face Area Elevation Conveyance Ratio=0.02
2D Face Min Length Ratio=0.05
2D Face Area Laminar Depth=0.2
2D Multiple Face Mann n=0
2D Composite LC=0

BC Line Name=DS Boundary
BC Line Storage Area=Perimeter 1
BC Line Start Position= 9522.59932215836 , 6644.19892020173
BC Line Middle Position= 9548.47627047713 , 6653.14803149531
BC Line End Position= 9574.35321879591 , 6662.09714278889
BC Line Arc= 2
9522.599322158366644.198920201739574.353218795916662.09714278889
LCMann Table=0
